--- DOGWAYFK.prj (project) ---

Proj Title=DOGWAYFK
Current Plan=p01
Default Exp/Contr=0,0
English Units
Geom File=g01
Flow File=f01
Plan File=p01
Background Map Layer=Inundation Boundary (01pct Value_0)
BEGIN DESCRIPTION:
----------MODEL BY WOOD PLC 2021----------
Stream Name: Dogway Fork
Flood Zone: Enhanced Approximate
Pocahontas County, WV
HEC-RAS Version: RAS 6.1
Vertical Datum: NAVD88
Projection: NAD 1983 StatePlane West Virginia S FIPS 4702 (US Feet)
Terrain: 1-meter LIDAR (FEMA Region III 3DEP collected 2016-2018)
Land Use: 2019 NLCD
Hydrologic Method:
WV SIR2010-5033 regression equations
Model Notes:
None
END DESCRIPTION:
DSS File=dss
DSS Export Rating Curves= 0
DSS Export Rating Curve Sorted= 0
DSS Export Volume Flow Curves= 0
DXF OffsetX= 0
DXF OffsetY= 0
DXF ScaleX= 0
DXF ScaleY= 0

--- DOGWAYFK.p01 (plan) ---

Plan Title=Floodplain
Program Version=6.00
Short Identifier=Floodplain
Geom File=g01
Flow File=f01
Subcritical Flow
K Sum by GR= 0
Std Step Tol= 0.01
Critical Tol= 0.01
Num of Std Step Trials= 20
Max Error Tol= 0.3
Flow Tol Ratio= 0.001
Split Flow NTrial= 30
Split Flow Tol= 0.02
Split Flow Ratio= 0.02
Log Output Level= 0
Friction Slope Method= 1
Unsteady Friction Slope Method= 2
Unsteady Bridges Friction Slope Method= 1
Parabolic Critical Depth
Global Vel Dist= 0 , 0 , 0
Global Log Level= 0
CheckData=True
Encroach Param=-1 ,0,0, 0
Computation Interval=0.1SEC
Output Interval=1SEC
Instantaneous Interval=Max Profile
Mapping Interval=1HOUR
Computation Time Step Use Courant=        0
Computation Time Step Use Time Series=    0
Computation Time Step Count To Double=0
Computation Time Step Max Doubling=0
Computation Time Step Max Halving=0
Computation Time Step Residence Courant=0
Run HTab= 0
Run UNet= 0
Run Sediment= 0
Run PostProcess= 0
Run WQNet= 0
Run RASMapper=-1
UNET Theta= 0
UNET Theta Warmup= 0
UNET ZTol= 0
UNET ZSATol= 0
UNET MxIter= 0
UNET Max Iter WO Improvement= 0
UNET MaxInSteps= 0
UNET DtIC= 0
UNET DtMin= 0
UNET MaxCRTS= 0
UNET WFStab= 0
UNET SFStab= 0
UNET WFX= 1
UNET SFX= 1
UNET Gravity=32.174
UNET 1D Methodology=Finite Difference
UNET DSS MLevel= 1
UNET Pardiso=0
UNET DZMax Abort= 0
UNET Use Existing IB Tables= 0
UNET Froude Reduction=False
UNET Froude Limit= 0
UNET Froude Power= 0
UNET D1 Cores= 0
UNET WindReference=Eulerian
UNET WindDragFormulation=Hsu (1988)
UNET D2 Coriolis=0
UNET D2 Cores= 0
UNET D2 Theta= 1
UNET D2 Theta Warmup= 1
UNET D2 Z Tol= 0.01
UNET D2 Volume Tol= 0.01
UNET D2 Max Iterations= 20
UNET D2 Equation= 0
UNET D2 RampUpFraction=0.1
UNET D2 TimeSlices= 1
UNET D2 Turbulence Formulation=Non-Conservative (original)
UNET D2 Eddy Viscosity=0.3
UNET D2 Transverse Eddy Viscosity=0.1
UNET D2 Smagorinsky Mixing=0
UNET D2 BCVolumeCheck=0
UNET D2 Cores=0
UNET D2 SolverType=PARDISO (Direct)
UNET D2 Minimum Iterations= 2147483647
UNET D2 Maximum Iterations= 2147483647
UNET D2 Restart Number= 10
UNET D2 Relaxation Coeff=1.3
UNET D2 SOR Precondition Iterations= 10
UNET D2 ILUT Maximum Fill= 8
UNET D2 ILUT Tolerance=1E-08
UNET D1D2 MaxIter= 0
UNET D1D2 ZTol=0.01
UNET D1D2 QTol=0.1
UNET D1D2 MinQTol=1
DSS File=dss
Write IC File= 0
Write IC File at Fixed DateTime=0
Write IC File at Sim End=0
Echo Input=False
Echo Parameters=False
Echo Output=False
Write Detailed= 0
HDF Write Warmup=0
HDF Write Time Slices=0
HDF Flush=0
HDF Compression= 1
HDF Chunk Size= 1
HDF Spatial Parts= 1
HDF Use Max Rows=0
HDF Fixed Rows= 1
Calibration Method= 0
Calibration Iterations= 20
Calibration Max Change=0.05
Calibration Tolerance=0.2
Calibration Maximum=1.5
Calibration Minimum=0.5
Calibration Optimization Method= 1
WQ AD Non Conservative
WQ ULTIMATE=-1
WQ Max Comp Step=1HOUR
WQ Output Interval=15MIN
WQ Output Selected Increments= 0
WQ Output face flow=0
WQ Output face velocity=0
WQ Output face area=0
WQ Output face dispersion=0
WQ Output cell volume=0
WQ Output cell surface area=0
WQ Output cell continuity=0
WQ Output cumulative cell continuity=0
WQ Output face conc=0
WQ Output face dconc_dx=0
WQ Output face courant=0
WQ Output face peclet=0
WQ Output face adv mass=0
WQ Output face disp mass=0
WQ Output cell mass=0
WQ Output cell source sink temp=0
WQ Output nsm pathways=0
WQ Output nsm derived pathways=0
WQ Create Restart=0
WQ Fixed Restart=0
WQ System Summary=0
WQ Write To DSS=0
Sorting and Armoring Iterations= 10
XS Update Threshold= 0.02
Bed Roughness Predictor= 0
Hydraulics Update Threshold= 0.02
Energy Slope Method= 1
Volume Change Method= 1
Sediment Retention Method= 0
Sediment TS Multiplier= 1
Warm Up Method= 0
XS Weighting Method= 0
Number of US Weighted Cross Sections= 1
Number of DS Weighted Cross Sections= 1
Upstream XS Weight=0
Main XS Weight=1
Downstream XS Weight=0
Number of DS XS's Weighted with US Boundary= 1
Upstream Boundary Weight= 1
Weight of XSs Associated with US Boundary= 0
Number of US XS's Weighted with DS Boundary= 1
Downstream Boundary Weight= 0.5
Weight of XSs Associated with DS Boundary= 0.5
Percentile Method= 0
Sediment Output Level= 3
Mass or Volume Output= 0
Output Increment Type= 1
Profile and TS Output Increment= 1
Transport Output Increment 1
XS Output Flag= 0
XS Output Increment= 10
Read HDF5 Sediment Hotstart= 0
Sediment Hotstart Type= 0
Write Gradation File= 0
Read Gradation Hotstart= 0
Write HDF5 File= 1
Write Binary Output= 1
Write DSS Sediment File= 0
DSS Sediment Output Type= 1
SV Curve= 0
Specific Gage Flag= 0
Subcell Erosion Methods= 0
Subcell Deposition Methods= 0
Advection Scheme= 1
Matrix Solver= 0
Implicit Weighting Factor= 1
Maximum Outer Loop Convergence Iterations= 5
Convergence Maximum Absolute= 0.001
Convergence RMSE= 0.0001
Grain Fractions Max Abs Error= 0.001
Max Subgrid Regions= 1
Max Subgrid Length Scale= 3.402823E+38
Initial Layer Thickness= 3.402823E+38
Min Layer Thickness= 3.402823E+38
Max Layer Thickness= 3.402823E+38
Number of Layers= 5

--- DOGWAYFK.f01 (steady flow) ---

Flow Title=Flow
Program Version=6.00
Number of Profiles= 6
Profile Names=01pct,10pct,04pct,02pct,0_2pct,01plus
River Rch & RM=DOGWAYFK,Main            ,22970
     629     333     443     533     877     930
River Rch & RM=DOGWAYFK,Main            ,18142
     766     409     542     650    1060    1130
River Rch & RM=DOGWAYFK,Main            ,17525
     858     461     608     729    1190    1270
River Rch & RM=DOGWAYFK,Main            ,14244
     969     523     688     824    1340    1430
River Rch & RM=DOGWAYFK,Main            ,10893
    1130     615     807     965    1560    1680
River Rch & RM=DOGWAYFK,Main            ,6193
    1260     686     899    1070    1730    1860
Boundary for River Rch & Prof#=DOGWAYFK,Main            , 1
Up Type= 0
Dn Type= 3
Dn Slope=0.01367
Boundary for River Rch & Prof#=DOGWAYFK,Main            , 2
Up Type= 0
Dn Type= 3
Dn Slope=0.01367
Boundary for River Rch & Prof#=DOGWAYFK,Main            , 3
Up Type= 0
Dn Type= 3
Dn Slope=0.01367
Boundary for River Rch & Prof#=DOGWAYFK,Main            , 4
Up Type= 0
Dn Type= 3
Dn Slope=0.01367
Boundary for River Rch & Prof#=DOGWAYFK,Main            , 5
Up Type= 0
Dn Type= 3
Dn Slope=0.01367
Boundary for River Rch & Prof#=DOGWAYFK,Main            , 6
Up Type= 0
Dn Type= 3
Dn Slope=0.01367
DSS Import GetInterval= 0
DSS Import GetPeak= 0
DSS Import FillOption= 0

--- DOGWAYFK.g01 (geometry) ---

Geom Title=Geometry
Program Version=6.10

River Reach=DOGWAYFK        ,Main
Reach XY= 30
     2164950.613      446653.3372163801.95724634 447098.07869053
     2163547.514      447513.5232162554.25117447447446.067857559
     2162015.379       446951.06  2162059.234706446669.635125486
      2161582.75      445961.473     2160958.739      445931.088
       2160159.6      446406.859     2159340.716      446176.299
     2159145.969       445898.73     2158698.145      446015.393
2158437.84222639445612.6084367872157048.26746492445146.843958986
     2156282.363      444270.307     2155105.722       443797.42
     2154243.996      445111.7982153778.13375967445160.178939917
 2153839.1837025445748.6549150822153414.04812147446060.335261326
       2153431.9      446597.334     2152940.849      447035.086
2153039.33855612447343.475911883 2152323.8537746447921.465174876
2152460.55023467448501.096382666     2152207.493      448800.901
     2152505.102      449446.061     2152181.381      449774.565
     2152517.157      450593.991 2152269.1921891 451031.64532569

Type RM Length L Ch R = 1 ,22970   ,187.9,187.3,185.3
XS GIS Cut Line= 3
2164903.98295056446476.2089429412164920.44688453446618.055543548
2165047.78889073446776.363821809
#Sta/Elev= 30
       0 3895.38       9 3894.18    17.1 3894.01    29.2  3893.1    41.2 3893.53
    53.3 3892.81    65.4 3891.39    77.5 3890.69    85.5 3888.96    89.6 3888.46
    97.6 3888.56   125.8 3886.98   133.9 3887.28   146.8 3885.92   162.2 3886.05
   167.9 3885.28     179 3883.09   187.5 3882.69   199.8 3882.65 204.4753882.975
   228.9 3889.07   231.7 3889.46   244.3 3888.81   249.5 3888.83   255.8 3889.53
   264.3 3891.46     270 3892.16   295.6 3892.19   331.6 3894.82     346  3896.9
#Mann= 6 ,-1,0
       0     .12       0      60      .1       0     100     .12       0
     179    .045       0 204.475     .12       0   332.8      .1       0
Bank Sta=179,204.475
XS Rating Curve= 0 ,0
Exp/Cntr(USF)=0,0
Exp/Cntr=0.3,0.1

Type RM Length L Ch R = 1 ,22783   ,135.8,134.6,134.3
XS GIS Cut Line= 3
2164769.39757165446533.9442598392164751.18560027446639.602015659
2164851.75855863446765.237322599
#Sta/Elev= 30
       0 3892.01     7.3  3890.9    15.5 3890.79      35  3889.8    60.1 3888.95
    72.3 3889.02    84.5 3888.09    92.6 3888.02   107.2 3886.52   119.5 3886.42
   123.3 3885.68   131.8 3882.39   134.9 3881.43   145.1 3881.21   150.2 3880.55
   153.6 3879.32   157.4 3877.04160.10583876.266   165.6    3876   174.5 3876.35
     188 3878.94   196.3 3880.24   206.6 3883.27     220 3885.95   227.1 3886.16
   243.2  3887.3   254.2 3886.16   257.8 3886.26   262.9 3886.82   268.1 3886.75
#Mann= 5 ,-1,0
       0      .1       0  147.22     .12       0160.1058    .045       0
   174.5     .12       0  207.22      .1       0
#XS Ineff= 2 , 0
          107.19 3892.86
Permanent Ineff=
       F       F
Bank Sta=160.1058,174.5
XS Rating Curve= 0 ,0
Exp/Cntr(USF)=0,0
Exp/Cntr=0.3,0.1

Type RM Length L Ch R = 1 ,22648   ,206.4,213.7,218.3
XS GIS Cut Line= 2
2164580.88731997446607.7970331552164809.98936574446926.067103774
#Sta/Elev= 30
       0 3901.82    11.9 3899.98    23.4 3895.91      51 3889.01    67.2 3884.49
    77.9 3883.66    89.3 3881.86    94.6 3880.26   106.5 3875.56   115.1    3874
   139.7 3875.85   149.6 3876.06   164.3 3875.31     189 3876.09   198.8 3875.29
   215.4 3875.64227.19833872.766   235.5 3872.06236.4926 3872.06   244.1 3872.38
   269.9 3880.97   277.7 3883.05   286.3 3884.37   317.1 3887.08   331.9 3886.43
   341.8 3887.11   347.2 3886.83   366.4 3887.33   376.3 3886.81   392.2 3888.03
#Mann= 5 ,-1,0
       0      .1       0      60     .12       0227.1983    .045       0
236.4926      .1       0     320     .12       0
#XS Ineff= 2 , 0
          169.59 3881.92
Permanent Ineff=
       F       F
Bank Sta=227.1983,236.4926
XS Rating Curve= 0 ,0
Exp/Cntr(USF)=0,0
Exp/Cntr=0.3,0.1

Type RM Length L Ch R = 1 ,22434   ,158.7,159.8,147.3
XS GIS Cut Line= 2
2164511.92413143446622.5862465042164525.66410031446980.714629957
#Sta/Elev= 30
       0 3904.58    10.5 3903.21    38.6 3900.91    54.6 3898.52    78.7  3892.8
    98.7 3885.73   106.7  3881.8   118.7 3874.13   122.7 3872.16   126.7 3871.44
   138.7 3870.12   154.7 3870.32   170.7 3869.67   182.7 3870.16   198.7 3869.62
   214.8 3869.84   222.8 3869.41   231.4 3868.05   234.8 3867.11   242.8  3866.8
   246.8 3866.84   250.8 3868.04   262.8 3874.86   270.8 3877.52   274.8 3878.02
   294.8 3877.74   310.8 3876.72   326.8 3876.72   334.8 3876.06   358.4 3875.29
#Mann= 5 ,-1,0
       0      .1       0     140     .12       0   231.4    .045       0
   250.8      .1       0     340     .12       0
#XS Ineff= 2 , 0
          164.67 3880.53
Permanent Ineff=
       F       F
Bank Sta=231.4,250.8
XS Rating Curve= 0 ,0
Exp/Cntr(USF)=0,0
Exp/Cntr=0.3,0.1

Type RM Length L Ch R = 1 ,22275   ,170.2,171,170.8
XS GIS Cut Line= 2
2164302.56263566446744.5220936972164458.80135972 446999.91231573
#Sta/Elev= 30
       0 3909.48    24.2 3905.67    33.7  3904.5    52.4 3899.49    66.4 3895.17
    75.8  3893.8    77.3 3893.28    80.2 3891.89    94.6 3883.24   108.6 3874.09
   115.1  3870.2     118 3868.69   125.7 3865.61     130 3864.25   132.1 3863.76
   135.5 3863.62   144.2 3863.88   148.7 3864.52   164.9 3867.71   169.6 3867.93
     179 3867.73   197.7 3870.68   207.1 3871.51   217.7 3874.16   225.8 3875.21
   230.5 3875.35   240.2 3874.36   277.4 3874.07     287 3873.43   299.4 3873.27
#Mann= 6 ,-1,0
       0     .06       0      30      .1       0     130    .045       0
   148.7     .12       0     230      .1       0     260     .12       0
Bank Sta=130,148.7
XS Rating Curve= 0 ,0
Exp/Cntr(USF)=0,0
Exp/Cntr=0.3,0.1

Type RM Length L Ch R = 1 ,22104   ,189.4,198.4,206.7
XS GIS Cut Line= 2
2164179.37441091446867.710318443  2164328.602423447079.033208046
#Sta/Elev= 30
       0 3892.51     7.4 3891.29    21.7 3888.03    27.5 3887.23    36.1 3885.19
    56.9 3881.75    70.4 3879.16    76.2 3877.06    91.5 3874.11    98.5 3872.33
   109.5 3868.66   119.4 3864.56   127.9 3862.61   138.9  3860.6   143.8 3860.11
   150.9 3859.93   159.5 3860.04   163.4 3860.69   168.3 3863.34   173.2 3864.87
   179.6 3865.07   188.2 3864.96   199.7 3865.98   202.8 3866.43   222.6 3871.37
   225.5 3871.69     237  3871.3   242.7 3870.57   248.5 3870.71   258.7  3870.4
#Mann= 3 ,-1,0
       0     .12       0   138.9    .045       0   163.4     .12       0
Bank Sta=138.9,163.4
XS Rating Curve= 0 ,0
Exp/Cntr(USF)=0,0
Exp/Cntr=0.3,0.1

Type RM Length L Ch R = 1 ,21905   ,187,180.5,172.6
XS GIS Cut Line= 2
2164088.23515521446914.7822417192164081.22444323447202.221432792
#Sta/Elev= 30
       0 3885.84    10.6 3883.01    18.4 3881.38    25.8 3878.64    54.4 3870.38
    70.4 3868.58    78.4 3868.34    86.4 3868.85    90.4 3868.34    94.4 3867.25
   106.4 3861.14   110.4 3859.62   118.4 3858.82   133.6 3855.52   139.1 3855.25
     150 3855.57   158.4 3858.41   162.4 3858.88   178.7  3858.8   198.5 3857.59
   226.5 3858.45   238.5 3860.83   246.5 3861.58   250.5 3862.44   254.5  3864.4
   258.5 3865.61   262.5 3865.85   270.5 3865.63   282.5 3863.46   287.5 3863.17
#Mann= 4 ,-1,0
       0     .06       0      50     .12       0   133.6    .045       0
     150     .12       0
#XS Ineff= 2 , 0
                          170.81          3869.5
Permanent Ineff=
       F       F
Bank Sta=133.6,150
XS Rating Curve= 0 ,0
Exp/Cntr(USF)=0,0
Exp/Cntr=0.3,0.1

Type RM Length L Ch R = 1 ,21725   ,230.9,233.6,231.3
XS GIS Cut Line= 3
2163890.81088841446976.9397215562163896.95200428447054.471309318
2164008.25972928447243.310622084
#Sta/Elev= 30
       0 3879.65     8.9 3875.33    12.3 3874.14    40.4 3868.06    60.4 3861.35
    75.9 3857.01    90.2 3855.72   104.1 3855.48   118.1 3856.05   122.7 3855.44
   127.3 3853.96   132.53852.913   137.6 3852.32   149.3 3852.19     155 3852.88
   164.5 3854.19   178.5 3855.19   187.7  3856.9   192.4 3856.99   201.6  3856.3
   207.7 3856.38   210.9  3856.9     218 3859.46   231.1 3863.05   243.4 3864.65
   251.5 3864.69   265.3  3862.6   271.3 3862.23   285.2 3861.62     297 3861.98
#Mann= 4 ,-1,0
       0     .12       0   132.5    .045       0     155     .12       0
  207.77      .1       0
#XS Ineff= 2 , 0
                          191.71         3860.33
Permanent Ineff=
       F       F
Bank Sta=132.5,155
XS Rating Curve= 0 ,0
Exp/Cntr(USF)=0,0
Exp/Cntr=0.3,0.1

Type RM Length L Ch R = 1 ,21491   ,205.9,200,198.7
XS GIS Cut Line= 3
2163716.55672582447024.5333694892163807.90582427447181.899463461
2163878.52865669447288.601351568
#Sta/Elev= 30
       0 3884.79    14.6  3881.4    23.9  3880.2    32.4 3877.79    42.4 3874.27
    56.2 3870.95    60.9 3868.87    65.5 3865.91    70.1 3863.81    82.1 3860.76
    93.2 3856.08   102.8 3851.18   107.1 3850.22   116.4 3849.59   126.7 3851.09
   143.6 3854.24   153.4 3855.71   171.9 3856.45   181.1 3855.73   196.9 3856.38
   219.5 3855.03   224.9 3855.78   238.7 3856.75   248.2 3858.64   262.5 3858.89
   272.2  3860.3     277 3860.48   282.7  3860.2     301 3858.41   309.9 3858.04
#Mann= 4 ,-1,0
       0     .12       0   102.8    .045       0   126.7     .12       0
     160      .1       0
Bank Sta=102.8,126.7
XS Rating Curve= 0 ,0
Exp/Cntr(USF)=0,0
Exp/Cntr=0.3,0.1

Type RM Length L Ch R = 1 ,21291   ,202,203.4,200.8
XS GIS Cut Line= 3
2163603.71372185447146.5880472522163655.91320668447268.642725016
2163792.55303462447388.394484331
#Sta/Elev= 30
       0 3864.84    15.9 3859.89    24.6 3857.94    28.9  3856.7    35.8 3855.54
      55 3854.42    69.4 3853.12    81.1 3852.63    85.5 3852.64   102.9 3851.75
   115.9 3850.76   124.6 3849.83     139 3850.32   153.2 3849.88   154.4 3849.78
   157.8 3848.99     165 3846.71     176 3846.13     181 3846.12   191.6 3846.73
   202.2 3848.18   218.4 3849.32   226.9 3850.29   234.2 3850.28   248.9 3850.73
   263.7 3851.99     282 3852.26   297.7 3853.54   303.5 3854.26   314.4 3854.35
#Mann= 6 ,-1,0
       0     .12       0      70      .1       0     130     .12       0
     165    .045       0   191.6     .12       0  232.75      .1       0
Bank Sta=165,191.6
XS Rating Curve= 0 ,0
Exp/Cntr(USF)=0,0
Exp/Cntr=0.3,0.1

Type RM Length L Ch R = 1 ,21088   ,151.3,164.9,171.3
XS GIS Cut Line= 3
2163491.32310685447242.2826440912163517.36289419 447403.52901957
2163670.59702741447538.735607705
#Sta/Elev= 30
       0 3847.39       7 3845.78    15.1 3844.69    63.7 3842.18    76.5    3843
    96.1 3842.11   108.3 3838.88   112.3 3838.82   120.4 3840.63   132.3 3841.93
   148.8 3840.86   160.2 3841.71   177.8 3841.72   183.1 3841.22   211.8 3842.48
   220.4 3841.75   231.1 3839.36   254.3 3835.74     260    3835   268.4 3835.74
   279.9 3837.27   288.4 3840.29   300.4 3846.21   311.1 3849.81     317 3851.33
   327.1 3852.76   343.1 3856.15   347.9 3857.39   353.8 3860.08   367.7 3862.26
#Mann= 5 ,-1,0
       0     .12       0     120      .1       0   254.3    .045       0
   268.4      .1       0  323.34     .12       0
Bank Sta=254.3,268.4
XS Rating Curve= 0 ,0
Exp/Cntr(USF)=0,0
Exp/Cntr=0.3,0.1

Type RM Length L Ch R = 1 ,20923   ,229.7,227.2,219.4
XS GIS Cut Line= 4
2163399.18232086447246.2887652212163452.26342583 447419.55350409
2163447.68328498447559.7929517592163466.43839279447636.663855969
#Sta/Elev= 30
       0 3850.33    19.1 3847.81    28.1 3846.21    41.5 3845.97    61.6 3842.51
    85.3 3840.54    99.2 3839.97   107.6 3840.36   111.8 3840.18   120.2 3837.84
   124.3 3837.23   141.1 3838.77   178.7 3838.37   186.8 3838.69   199.4 3838.35
   210.9 3837.42   242.9 3836.72   254.9 3837.07   262.9 3835.45     272 3834.58
   278.9 3833.92   282.9 3834.45   294.9 3839.12   306.9 3840.09   314.9 3839.63
   318.9 3839.89   340.5 3843.11   355.9 3846.12     376 3851.43   400.7 3857.08
#Mann= 3 ,-1,0
       0      .1       0     272    .045       0   282.9      .1       0
Bank Sta=272,282.9
XS Rating Curve= 0 ,0
Exp/Cntr(USF)=0,0
Exp/Cntr=0.3,0.1

Type RM Length L Ch R = 1 ,20696   ,226.8,235.8,235.2
XS GIS Cut Line= 3
2163242.92316494447301.6512227762163296.65792873447595.657144684
2163338.11046081447677.794569343
#Sta/Elev= 30
       0 3836.97    15.8 3835.17    31.6 3835.21    60.5  3833.9    68.6 3833.91
    80.8 3832.73    84.9 3832.66    90.1 3833.12    96.9 3833.12   101.2 3832.32
   105.2 3830.81   109.3 3829.65   115.93828.963   117.4 3828.71   132.83829.709
   162.2 3829.59   227.2 3832.89   231.3 3832.77   243.5 3833.21   251.6 3832.75
   259.8 3832.62     272  3833.2   315.6 3837.94   335.4 3841.49   351.1 3844.96
   363.3 3846.56   371.1 3848.46     380 3850.04     386  3851.6   390.9 3852.56
#Mann= 5 ,-1,0
       0      .1       0   115.9    .045       0   132.8      .1       0
     260     .12       0  368.88      .1       0
Bank Sta=115.9,132.8
XS Rating Curve= 0 ,0
Exp/Cntr(USF)=0,0
Exp/Cntr=0.3,0.1

Type RM Length L Ch R = 1 ,20460   ,205.2,214.9,209.4
XS GIS Cut Line= 2
2163083.70028188447366.4723991192163085.70334244447697.683141177
#Sta/Elev= 30
       0 3825.83    11.1 3826.23    14.7 3826.07    22.7 3825.23    30.4 3825.58
    42.7 3825.45    50.7 3825.79    66.6 3824.53    70.7 3824.43    78.7 3824.62
    98.7 3823.97   110.9 3823.36   122.7 3822.07   134.7 3822.04   138.7  3821.8
   155.2 3821.51   170.7 3820.91   178.7 3821.06   182.1 3821.54     190 3823.71
   195.4  3824.1   207.5 3824.28   218.7 3824.13   226.7 3824.45   238.7 3824.04
   242.7 3824.14   266.7 3825.73   289.4 3825.88   314.7 3827.47   331.2 3829.42
#Mann= 5 ,-1,0
       0      .1       0   155.2    .045       0   182.1      .1       0
     190     .12       0     290      .1       0
Bank Sta=155.2,182.1
XS Rating Curve= 0 ,0
Exp/Cntr(USF)=0,0
Exp/Cntr=0.3,0.1

Type RM Length L Ch R = 1 ,20245   ,156.4,161.5,159.8
XS GIS Cut Line= 3
2162904.35438221447343.6710934212162891.40646764447480.646851322
2162858.25716349447712.663750483
#Sta/Elev= 30
       0 3824.56    21.6 3818.77    25.6  3817.9    29.6 3817.35    49.7 3816.56
    69.8 3816.86    73.8 3816.71    93.9 3818.25     114 3817.23     122 3817.61
     130 3818.37   134.1 3818.45   142.2    3818   150.2 3817.22   158.6 3817.18
   162.4 3816.73   172.7 3814.07178.4979 3813.29   190.4  3813.1194.6979 3813.28
   202.8 3814.69     223 3816.25   238.1 3816.32   255.3 3815.23   259.3 3815.25
   304.1  3817.6     328 3818.33   336.1 3818.93   348.2 3818.72     372 3820.13
#Mann= 3 ,-1,0
       0      .1       0178.4979    .045       0194.6979      .1       0
#XS Ineff= 2 , 0
           136.3 3820.97  261.75         3820.15
Permanent Ineff=
       F       F
Bank Sta=178.4979,194.6979
XS Rating Curve= 0 ,0
Exp/Cntr(USF)=0,0
Exp/Cntr=0.3,0.1

Type RM Length L Ch R = 1 ,20083   ,149.6,150.1,160.3
XS GIS Cut Line= 3
2162786.24578798447354.454035729 2162728.1570316447521.709592903
2162693.70919949447644.166167714
#Sta/Elev= 30
       0  3816.2    11.4 3813.74    15.6 3813.08    28.3  3811.7    36.8 3811.38
    45.2 3810.35    49.5 3810.07    91.9 3809.83   100.3 3809.13   113.8 3806.09
   121.4 3805.74   138.9 3806.01   146.9 3806.82   151.1 3807.47   155.3 3807.74
   172.3 3810.76   176.5 3811.04   180.7  3810.9   201.4 3808.66   209.7 3808.15
   225.3 3807.74     235 3808.19   238.8 3808.56   244.7 3808.68   259.6 3810.19
   272.1 3812.29   280.4 3812.66   284.5 3813.06   288.7  3813.8   304.3 3815.43
#Mann= 3 ,-1,0
       0      .1       0   113.8    .045       0   138.9      .1       0
Bank Sta=113.8,138.9
XS Rating Curve= 0 ,0
Exp/Cntr(USF)=0,0
Exp/Cntr=0.3,0.1

Type RM Length L Ch R = 1 ,19933   ,76.1,77.7,68.8
XS GIS Cut Line= 3
2162668.03901598447327.685551076 2162636.9606378447391.223568698
2162511.95649443447572.168792797
#Sta/Elev= 30
       0  3813.2    10.6 3810.67    19.5 3808.36    23.9 3807.63    28.4 3806.34
    36.9 3803.57    39.9 3803.14    41.7 3802.97    55.1 3804.23      64 3802.73
   116.9 3800.26   121.7 3799.96   131.4  3798.8   135.5 3798.55   141.2 3798.45
   164.7 3798.56   175.2 3798.35   177.7 3798.66   184.8 3800.08   191.7 3800.99
   204.4 3801.41   209.2 3802.48   222.2 3802.81     228 3803.13   233.7  3803.6
   243.3 3804.69     253 3804.24   262.7 3804.33   268.2 3804.12   290.7 3804.72
#Mann= 3 ,-1,0
       0      .1       0   131.4    .045       0   177.7      .1       0
Bank Sta=131.4,177.7
XS Rating Curve= 0 ,0
Exp/Cntr(USF)=0,0
Exp/Cntr=0.3,0.1

Type RM Length L Ch R = 1 ,19856   ,100.9,99.2,95.4
XS GIS Cut Line= 2
2162625.47230632447318.8320276742162456.59141488 447517.97749297
#Sta/Elev= 30
       0 3809.59     8.3 3807.21    14.4 3805.14    25.3 3802.12    28.1  3801.6
    34.5 3800.86    55.5 3797.01    62.2 3796.74   107.6 3796.32   113.2 3795.89
   116.1 3795.94   121.8 3796.83   123.7 3796.94   125.7 3796.79     136 3796.82
   144.7 3796.77   155.2  3795.7   187.5 3795.52   192.7 3795.54   195.6 3795.84
   201.2 3796.84   206.9 3797.49   212.6 3797.14   218.5 3797.42   224.6 3798.58
   230.8 3800.15     241 3801.92   243.2 3802.09   249.6 3801.65   261.1 3802.04
#Mann= 4 ,-1,0
       0     .12       0      50      .1       0   125.7    .045       0
     136      .1       0
#XS Ineff= 2 , 0
                           168.2         3801.57
Permanent Ineff=
       F       F
Bank Sta=125.7,136
XS Rating Curve= 0 ,0
Exp/Cntr(USF)=0,0
Exp/Cntr=0.3,0.1

Type RM Length L Ch R = 1 ,19756   ,105.9,106.6,105.9
XS GIS Cut Line= 2
2162546.20235795447259.3810923292162381.26523661447468.257840655
#Sta/Elev= 30
       0 3808.56     3.3 3806.97    31.2  3800.2      42 3798.07    48.5 3796.22
    51.1 3795.63    58.4 3794.98    67.8 3793.14    74.3 3790.28    79.6 3787.18
    87.2 3783.61    96.7 3781.07101.97733780.358   109.3 3780.44   124.6 3780.03
130.16163780.518   150.1 3784.32   160.3 3785.67   170.5 3787.71   179.3 3788.79
   185.8 3790.07     196 3791.14   201.1 3792.07   206.2 3793.38   221.4 3795.74
   231.6 3795.91   239.1 3796.35   244.8 3796.94     252  3798.2   266.1 3798.55
#Mann= 3 ,-1,0
       0     .12       0101.9773    .045       0130.1616      .1       0
Bank Sta=101.9773,130.1616
XS Rating Curve= 0 ,0
Exp/Cntr(USF)=0,0
Exp/Cntr=0.3,0.1

Type RM Length L Ch R = 1 ,19650   ,222.4,222.8,222.7
XS GIS Cut Line= 2
2162461.74997646447194.2091905322162315.52655521447384.499944203
#Sta/Elev= 30
       0 3802.24     2.6 3802.01     8.9 3799.84    18.9 3798.08    23.2 3796.91
    28.8 3795.82    35.4  3794.9    44.1 3794.33    59.2 3791.61      66 3789.67
    74.6 3788.71      86 3785.28    97.4  3780.4   104.6 3776.94   105.9 3776.56
   108.8 3776.32   114.7 3776.47   120.2 3776.88   127.3 3777.84   137.3 3780.85
     145 3782.62   153.6 3783.87   160.1 3785.03   170.2 3785.48   177.2 3786.04
     193 3786.58   210.6 3789.44   225.7 3790.46   230.8 3791.31     240 3792.47
#Mann= 5 ,-1,0
       0      .1       0      20     .12       0      80      .1       0
   104.6    .045       0   120.2      .1       0
Bank Sta=104.6,120.2
XS Rating Curve= 0 ,0
Exp/Cntr(USF)=0,0
Exp/Cntr=0.3,0.1

Type RM Length L Ch R = 1 ,19427   ,178.5,177,175.3
XS GIS Cut Line= 2
2162301.38522112447047.6979354322162136.13272451447247.002461646
#Sta/Elev= 30
       0 3785.85     8.2 3784.81    13.3 3784.49    21.8 3783.01    33.1 3782.04
      36  3781.5    45.8  3780.4    58.3 3777.93    77.1 3776.41    85.1 3775.15
      95  3773.2    98.5 3772.62     111 3771.47   114.7 3771.61   115.83771.799
   118.4 3772.68   121.4 3774.07   124.1 3774.84   126.6 3775.29     146  3776.5
   163.8 3778.01   171.1 3779.63     189 3782.76   209.3 3786.69   220.6 3789.48
   225.4 3790.23     232 3791.76   240.9 3793.33   245.4 3794.34   258.9 3797.88
#Mann= 3 ,-1,0
       0      .1       0      95    .045       0   115.8      .1       0
Bank Sta=95,115.8
XS Rating Curve= 0 ,0
Exp/Cntr(USF)=0,0
Exp/Cntr=0.3,0.1

Type RM Length L Ch R = 1 ,19250   ,176.9,196.6,208.5
XS GIS Cut Line= 3
2162269.45616222446930.8067262392162132.24651352446967.863346691
2162045.11337894447102.068404543
#Sta/Elev= 30
       0 3785.98     9.5 3784.49    13.8 3783.53    42.1 3773.51    46.9 3772.04
    55.2 3770.66    63.5 3768.88    67.6 3768.39    71.5 3768.36    74.7  3768.8
    88.3 3769.38   117.3 3771.55   125.6 3771.71   143.7 3770.76   148.5 3770.94
   156.9 3772.18   160.5 3772.28   167.5 3771.69   172.3 3771.74   181.8 3768.35
     187 3767.45   196.2 3766.86   206.7 3767.36     220 3769.41   224.8 3771.07
   234.3 3776.22   243.8 3780.51   258.8 3788.26   286.8 3793.96   302.1 3797.78
#Mann= 3 ,-1,0
       0      .1       0     187    .045       0   206.7      .1       0
#XS Ineff= 2 , 0
          162.04 3780.79
Permanent Ineff=
       F       F
Bank Sta=187,206.7
XS Rating Curve= 0 ,0
Exp/Cntr(USF)=0,0
Exp/Cntr=0.3,0.1

Type RM Length L Ch R = 1 ,19053   ,156.9,160.2,160.1
XS GIS Cut Line= 3
 2162196.3444516446804.6139106462162073.15622685446868.711848725
2161945.96188098446861.701136748
#Sta/Elev= 30
       0 3780.39     9.4 3776.46    18.6 3772.99    31.8 3767.42    35.9 3766.86
      45 3766.48    58.8 3766.86    67.8 3766.15    76.8 3765.99    83.7 3765.21
    99.4 3764.63   104.4 3764.77   113.2 3765.72   139.8 3765.92   147.9 3766.29
   151.9 3765.53   171.9 3763.62   179.9 3761.14   183.43760.358   188.7 3759.88
   199.8 3759.58   203.1 3760.17     208 3762.25     224 3770.53     232  3775.7
     240 3781.25     244 3783.04     248 3783.74     256 3784.13   266.3 3785.47
#Mann= 3 ,-1,0
       0      .1       0   183.4    .045       0   203.1      .1       0
Bank Sta=183.4,203.1
XS Rating Curve= 0 ,0
Exp/Cntr(USF)=0,0
Exp/Cntr=0.3,0.1

Type RM Length L Ch R = 1 ,18893   ,130.1,124,116.2
XS GIS Cut Line= 3
2162182.71497812446728.603982199 2162028.6214283 446712.60077858
2161839.92543969446762.183282455
#Sta/Elev= 30
       0 3784.02    14.6 3782.37    26.7 3779.17    46.8 3776.16    50.8 3775.15
    62.9 3771.22      79 3764.03      91 3762.11      95 3760.43   103.1 3756.08
   107.1 3754.99   114.7 3754.39   123.2 3754.62     1293755.535   143.3 3759.91
   147.3 3760.42   184.3 3758.56     205 3758.37   221.3 3760.08     234 3760.27
   246.4 3759.85     254 3760.59   271.2 3765.39   283.5    3770   296.6 3778.73
   304.3 3782.74   308.4  3784.2   316.2 3786.55   328.6 3789.52     350 3794.11
#Mann= 3 ,-1,0
       0      .1       0   107.1    .045       0     129      .1       0
#XS Ineff= 1 ,-1
  151.98     339 3770.78
Permanent Ineff=
       F
Bank Sta=107.1,129
XS Rating Curve= 0 ,0
Exp/Cntr(USF)=0,0
Exp/Cntr=0.3,0.1

Type RM Length L Ch R = 1 ,18769   ,123.1,122.4,122.6
XS GIS Cut Line= 3
2162104.77378723446556.4795458712161977.30213297 446629.82915698
2161850.54261086446673.981350076
#Sta/Elev= 30
       0  3777.7    18.5 3774.82    36.1 3771.09    42.2 3769.23    49.5 3765.89
    57.5 3761.65    65.3 3758.27    88.8 3749.29    91.8 3748.55   106.8 3747.86
   111.4 3748.63   126.9 3754.69   129.8 3755.58   134.5 3755.93   148.3 3755.87
   165.2 3756.62   177.9 3755.82   200.8 3756.49   207.6 3756.24   216.6  3756.4
   228.7 3755.56   238.5 3755.45     248 3756.12   249.9 3756.52   254.2 3758.21
   263.7 3763.83   271.1 3767.83   275.3 3770.54   279.4 3773.55   281.3 3774.29
#Mann= 3 ,-1,0
       0      .1       0    91.8    .045       0   111.4      .1       0
Bank Sta=91.8,111.4
XS Rating Curve= 0 ,0
Exp/Cntr(USF)=0,0
Exp/Cntr=0.3,0.1

Type RM Length L Ch R = 1 ,18647   ,213,212.8,210.9
XS GIS Cut Line= 2
2162046.11490922446445.0645392352161861.83333725446562.243582286
#Sta/Elev= 30
       0 3771.47     7.3 3769.71    13.1 3768.97    21.3 3767.09    30.5 3766.01
    35.5 3764.56      45 3761.19    59.9 3755.64    63.9  3753.9    68.1 3752.64
    78.1 3750.71    91.3  3747.7    97.1 3747.03   106.6 3744.42   111.6 3743.73
   114.5 3743.43   120.8 3743.11   130.3 3743.15   134.4 3743.63     135 3743.81
   141.9 3747.62   144.5 3748.65   149.2 3749.66     154 3750.23   164.2 3750.44
   171.7 3749.82     184 3749.34   187.2 3749.44   210.1 3751.48   218.4  3751.7
#Mann= 3 ,-1,0
       0      .1       0   111.6    .045       0   134.4      .1       0
Bank Sta=111.6,134.4
XS Rating Curve= 0 ,0
Exp/Cntr(USF)=0,0
Exp/Cntr=0.3,0.1

Type RM Length L Ch R = 1 ,18434   ,185,191.1,193.6
XS GIS Cut Line= 2
2161920.92362391446266.7921489532161742.65123363446396.991085676
#Sta/Elev= 30
       0 3756.55    24.4 3754.37    36.6 3753.82      48  3752.9    65.1 3751.87
    70.3 3750.08    75.2 3746.96    80.2 3744.52    88.1 3739.87      91 3738.46
    92.2 3738.07      99 3736.84   108.2 3735.76   114.9 3735.22     1273735.824
   129.7  3736.2   139.6 3738.37   154.5 3740.04   159.4  3741.2   164.4 3742.04
   169.3 3743.31   173.6 3744.92   179.7 3748.41   185.4 3750.59     194 3752.78
   199.1 3753.45     204 3753.51     209 3754.27   213.9  3755.8   220.8 3757.53
#Mann= 3 ,-1,0
       0      .1       0   108.2    .045       0     127      .1       0
Bank Sta=108.2,127
XS Rating Curve= 0 ,0
Exp/Cntr(USF)=0,0
Exp/Cntr=0.3,0.1

Type RM Length L Ch R = 1 ,18243   ,100.5,100.9,101.5
XS GIS Cut Line= 3
2161923.92821476446021.4172297452161763.68336956446175.652893248
2161619.46300889446230.737058784
#Sta/Elev= 30
       0 3762.25     5.3 3761.24    16.3 3760.21    22.7 3759.21    50.6 3753.38
    59.1 3751.13    71.8 3748.48    81.7 3746.06   104.3 3743.38   152.4 3742.02
   160.9 3742.61   182.9 3741.09     190 3741.38   200.5 3740.58   213.1 3741.43
   226.2 3741.68   238.7 3739.71   251.9 3735.73   264.7 3733.22     269 3731.93
   277.5 3728.27   281.8 3727.14   290.4 3726.45     299 3726.24   303.8 3726.87
   322.4 3732.25   347.1 3743.29   362.6 3749.01   371.3 3751.48   376.8 3753.39
#Mann= 3 ,-1,0
       0      .1       0   281.8    .045       0   303.8      .1       0
Bank Sta=281.8,303.8
XS Rating Curve= 0 ,0
Exp/Cntr(USF)=0,0
Exp/Cntr=0.3,0.1

Type RM Length L Ch R = 1 ,18142   ,126.4,118.5,113.2
XS GIS Cut Line= 4
2161868.34591453445941.909503272 2161712.3889744446090.032989784
2161616.96326674446122.7910685332161579.22026297446149.852090107
#Sta/Elev= 30
       0 3748.84     5.8 3749.19    16.8 3748.79    36.4 3747.18    44.9  3746.1
    55.4 3744.13      94 3740.06   115.1 3739.67   127.1 3738.31   138.2 3738.57
     150 3737.68   169.4 3736.33   184.8 3734.79   202.2  3734.2     209 3733.43
   223.8 3728.78   236.6 3721.89   240.7  3720.2   244.9 3719.55   261.7 3719.44
     265 3719.84   274.4 3724.72   278.8 3725.57   304.1 3725.64     317 3726.78
     324 3729.14   331.7 3732.44   340.7 3735.51   354.4 3739.28   362.4 3740.54
#Mann= 4 ,-1,0
       0     .12       0     150      .1       0   240.7    .045       0
     265      .1       0
Bank Sta=240.7,265
XS Rating Curve= 0 ,0
Exp/Cntr(USF)=0,0
Exp/Cntr=0.3,0.1

Type RM Length L Ch R = 1 ,18023   ,224,213.7,208.3
XS GIS Cut Line= 3
2161777.70479352445841.1417788992161661.52728075445966.333064209
2161533.33140459446081.509046694
#Sta/Elev= 30
       0 3743.89    16.4 3742.83    27.3 3741.17    54.6 3740.11      69 3740.77
   100.2 3738.21     114 3738.22   122.8 3737.18   131.6 3737.58   136.5 3737.02
   143.4 3735.09   159.6 3734.33   170.8 3733.13     178 3732.07   183.4    3730
     187 3727.82     193 3722.86   199.5 3718.28     205 3715.55   210.6 3715.06
   228.9  3715.6   247.9 3720.49   252.9 3720.71     264 3720.08   274.8 3720.46
   295.6 3719.78   306.9 3720.44   315.4 3722.85   324.7 3727.28   343.1 3730.74
#Mann= 9 ,-1,0
       0      .1       0      30     .12       0      60      .1       0
     170     .12       0  190.79      .1       0     205    .045       0
   228.9      .1       0  310.79     .12       0  340.79      .1       0
Bank Sta=205,228.9
XS Rating Curve= 0 ,0
Exp/Cntr(USF)=0,0
Exp/Cntr=0.3,0.1

Type RM Length L Ch R = 1 ,17810   ,140.3,142.4,143.9
XS GIS Cut Line= 2
2161517.26960763445774.0486520262161387.53853504446063.448737037
#Sta/Elev= 30
       0 3738.36    12.3 3733.43    25.3 3729.76    36.5 3727.68    45.6 3725.14
    51.6 3723.22    60.4 3718.89      78 3713.91   117.4 3714.22   130.6 3712.41
   139.4 3712.36   148.1  3710.3   151.5 3710.06   161.2 3711.26   178.7 3710.34
   187.8 3711.17   191.9 3710.81   198.2 3708.41   205.1 3707.44   218.2  3707.7
   221.1 3708.22   224.1 3709.37   235.8 3716.27   240.1 3718.25   244.5 3718.96
   257.7 3718.12   279.6 3718.56   292.7 3719.89   301.5 3721.97   317.1 3727.52
#Mann= 5 ,-1,0
       0     .06       0      10      .1       0   198.2    .045       0
   221.1      .1       0     230     .12       0
#XS Ineff= 2 , 0
          171.51 3715.83
Permanent Ineff=
       F       F
Bank Sta=198.2,221.1
XS Rating Curve= 0 ,0
Exp/Cntr(USF)=0,0
Exp/Cntr=0.3,0.1

Type RM Length L Ch R = 1 ,17667   ,150.7,142.1,136.1
XS GIS Cut Line= 3
2161378.40442821445769.2748444882161292.06343168445953.855595748
2161293.37642088446017.240846168
#Sta/Elev= 30
       0 3728.59     4.3 3728.12    13.1 3725.68    16.6 3725.08    34.7 3722.93
    46.7 3719.33    55.8 3717.49    79.4 3712.05    88.2 3708.53    91.9  3707.6
    99.7  3704.9   106.9 3703.11   112.9 3702.26   123.5 3701.49   127.9 3702.27
     137  3705.3   145.6 3706.21     150 3706.32   158.9 3705.71   163.3 3705.93
   173.1 3705.34   185.4 3705.45   189.8 3705.66   198.6 3706.74   215.1 3707.45
   226.7  3709.2   235.1  3709.7   255.1 3714.68   263.1 3716.02   267.2 3716.37
#Mann= 4 ,-1,0
       0     .12       0      30      .1       0   112.9    .045       0
   127.9      .1       0
#XS Ineff= 2 , 0
                          147.47         3708.95
Permanent Ineff=
       F       F
Bank Sta=112.9,127.9
XS Rating Curve= 0 ,0
Exp/Cntr(USF)=0,0
Exp/Cntr=0.3,0.1

Type RM Length L Ch R = 1 ,17525   ,106.5,101.9,100.7
XS GIS Cut Line= 2
2161174.08204206445773.5132726342161212.44381775 446015.60162162
#Sta/Elev= 30
       0 3725.87    15.9 3724.99    19.9 3724.19    22.5  3723.2      28 3721.72
      40 3717.49    44.2 3715.55    48.3 3713.13    68.5 3699.72    72.6 3697.56
75.634113696.899    88.8 3696.11    92.8 3696.16    96.9 3696.65   100.9 3697.15
     109 3699.98   113.4 3700.45   117.1  3700.6   127.4 3700.04   141.4  3700.1
   149.5 3699.58   157.6 3700.31   173.8 3702.81   177.9 3703.07     190 3703.34
   206.2 3702.66   214.8  3703.1   221.8 3703.91   234.6 3706.66   245.1  3707.2
#Mann= 3 ,-1,0
       0      .1       075.63411    .045       0    96.9      .1       0
#XS Ineff= 2 , 0
                          116.74         3704.67
Permanent Ineff=
       F       F
Bank Sta=75.63411,96.9
XS Rating Curve= 0 ,0
Exp/Cntr(USF)=0,0
Exp/Cntr=0.3,0.1

Type RM Length L Ch R = 1 ,17423   ,180.3,176.8,173.5
XS GIS Cut Line= 3
2161065.61676268445821.1111732492161107.68103454445939.291746582
 2161138.7284733446066.486092457
#Sta/Elev= 30
       0 3715.05     8.6 3712.09    14.6 3709.36    20.8 3706.01    28.9 3702.53
      34 3699.99    38.3 3698.51    43.4 3697.44    59.5 3696.21    67.8 3692.93
      75 3690.63    76.5 3690.21    89.2 3690.03    93.5 3690.75     102 3695.05
   105.4 3696.15     119  3698.2   127.4 3697.57   135.6 3698.27     148 3699.82
   156.2    3700   180.9 3699.64   189.1 3698.82   193.3 3698.76   205.6 3699.97
   213.9 3700.41     218 3701.27   230.3 3707.07   246.8 3713.87   256.4 3718.38
#Mann= 3 ,-1,0
       0      .1       0      75    .045       0    93.5      .1       0
Bank Sta=75,93.5
XS Rating Curve= 0 ,0
Exp/Cntr(USF)=0,0
Exp/Cntr=0.3,0.1

Type RM Length L Ch R = 1 ,17246   ,200,199.3,198.1
XS GIS Cut Line= 3
2160868.31529703445840.1402486162160953.44537104446004.391214943
2161033.56779364446112.556485451
#Sta/Elev= 30
       0 3709.93     3.6 3708.35    14.7 3700.13    24.4 3694.33    27.4 3693.04
    33.3 3691.35    41.7  3690.7    54.1 3690.95    65.9 3691.77    80.8 3693.56
    91.3 3693.73    95.8 3693.05   104.5 3687.23   107.5 3685.95   112.7 3685.48
   137.2 3686.03   158.9 3691.76   164.9 3691.99   181.4 3691.28   195.9 3691.69
   210.9 3691.07   235.8 3692.17   244.7  3693.1   250.7 3692.87   255.7 3693.23
   270.6 3698.14   281.9 3703.97   300.5 3715.41   313.3 3724.24   319.6 3727.09
#Mann= 3 ,-1,0
       0      .1       0   107.5    .045       0   137.2      .1       0
Bank Sta=107.5,137.2
XS Rating Curve= 0 ,0
Exp/Cntr(USF)=0,0
Exp/Cntr=0.3,0.1

Type RM Length L Ch R = 1 ,17047   ,200.7,199.6,198.4
XS GIS Cut Line= 2
2160686.03678562 445930.277974042160827.25255545446178.657484095
#Sta/Elev= 30
       0 3700.61    12.5 3699.94    35.5 3700.28    50.6 3698.55    63.2 3697.53
    69.1 3696.34    86.2 3689.82    94.6 3685.73     100 3683.86   113.8 3683.49
   127.6 3680.28   136.8 3679.84     146 3680.14     168 3683.51   176.8 3683.12
   191.4  3681.7   201.2 3682.45     215 3682.69   224.2 3682.32   228.8 3682.91
   233.4 3684.52   238.4 3687.01   242.6 3690.67   247.3 3696.49   251.8 3700.24
   256.4 3702.95   265.6 3706.38   273.6 3708.86   279.4 3711.62   285.7  3713.2
#Mann= 3 ,-1,0
       0      .1       0   127.6    .045       0     146      .1       0
#XS Ineff= 2 , 0
                          171.03         3691.69
Permanent Ineff=
       F       F
Bank Sta=127.6,146
XS Rating Curve= 0 ,0
Exp/Cntr(USF)=0,0
Exp/Cntr=0.3,0.1

Type RM Length L Ch R = 1 ,16848   ,228.5,229,231.2
XS GIS Cut Line= 2
2160501.75521364446032.4340628532160653.98781658446256.776846129
#Sta/Elev= 30
       0  3687.3    25.1 3686.39    34.7 3686.55    49.2 3686.25    73.4 3685.11
    77.2 3684.22    82.7 3681.62    87.9 3676.96    89.8 3675.72    92.7  3674.4
    94.4 3674.35   107.2 3675.83   121.7 3676.42   125.4 3676.16   131.9 3673.74
   134.7  3673.1   139.7 3672.54   153.9 3673.11   157.8 3673.67   174.9  3677.6
   179.8 3677.82   184.6  3677.2   194.3 3677.23   199.1 3677.55   203.9 3678.54
   229.8 3688.99   237.8 3693.06   252.3 3701.13   264.3 3706.66   271.1 3709.21
#Mann= 3 ,-1,0
       0      .1       0   134.7    .045       0   153.9      .1       0
#XS Ineff= 2 , 0
          116.59 3685.54  178.79          3685.5
Permanent Ineff=
       F       F
Bank Sta=134.7,153.9
XS Rating Curve= 0 ,0
Exp/Cntr(USF)=0,0
Exp/Cntr=0.3,0.1

Type RM Length L Ch R = 1 ,16619   ,148.4,145.7,144.8
XS GIS Cut Line= 2
2160321.98954595446123.2374711272160453.19001295446361.601678357
#Sta/Elev= 30
       0 3675.79    11.9 3676.11    20.5 3675.87    43.3 3674.09    53.1 3672.84
    61.6 3672.54    75.3 3672.73    84.4 3673.38      89 3673.35    98.1 3669.84
   106.1 3665.72   107.2 3665.36   111.8 3664.99   120.7 3665.36   123.8 3666.05
   130.1 3667.88   135.6 3668.54   148.3 3668.99   157.5 3669.78   170.4 3669.87
   179.7 3671.26   198.5 3671.26     218 3675.06   223.9 3676.92   235.7 3681.68
   239.6 3682.72   244.2 3684.91   253.4 3690.86   259.2 3695.33   272.1 3701.69
#Mann= 4 ,-1,0
       0     .12       0      60      .1       0   106.1    .045       0
   123.8      .1       0
Bank Sta=106.1,123.8
XS Rating Curve= 0 ,0
Exp/Cntr(USF)=0,0
Exp/Cntr=0.3,0.1

Type RM Length L Ch R = 1 ,16473   ,197.6,211.4,234.3
XS GIS Cut Line= 3
2160225.33285567446120.5687277112160232.34356765446272.801330648
2160333.49812618446405.003327936
#Sta/Elev= 30
       0 3671.95     8.6 3672.38    32.6 3672.27    36.6 3672.69    52.7 3672.87
    60.7 3672.22    72.7 3670.19      76 3670.03    88.7 3669.67   128.7 3670.15
   144.8 3668.34   158.7 3669.14     168 3668.45   183.1 3665.12   198.2 3662.31
   211.4 3661.95   219.7 3662.26   223.4  3662.7   232.4 3664.81   243.9 3664.45
   253.6 3666.66   268.7 3667.61   277.2 3669.76   283.8 3672.76   288.9  3676.1
   295.2 3681.49   303.5 3689.46   310.1 3694.35     314 3696.74   318.9 3698.18
#Mann= 5 ,-1,0
       0      .1       0      60     .12       0   198.2    .045       0
   219.7     .12       0  242.39      .1       0
Bank Sta=198.2,219.7
XS Rating Curve= 0 ,0
Exp/Cntr(USF)=0,0
Exp/Cntr=0.3,0.1

Type RM Length L Ch R = 1 ,16261   ,148.5,145.8,145.6
XS GIS Cut Line= 3
2160184.27011409446135.5916819482160181.26552324446291.830406016
 2160058.0772985446429.040054716
#Sta/Elev= 30
       0  3670.3    29.6  3671.1    49.6 3670.25    64.5 3669.05    89.6 3669.02
   113.6 3667.93   125.6 3666.66     139 3665.99   150.8 3664.25   175.9 3662.87
   180.7 3661.98   189.2 3658.29     192 3658.06   197.7 3658.32   211.8 3660.47
     243 3659.84   254.8 3661.72   260.2 3662.05   271.3 3658.38   276.3 3657.33
   279.8 3657.28   292.5  3657.5   297.8  3658.2   301.6 3659.46   308.1 3662.97
     314 3665.42   324.7 3671.85   331.5 3678.02   335.5 3680.62   340.7 3682.85
#Mann= 4 ,-1,0
       0     .12       0      40      .1       0   276.3    .045       0
   292.5      .1       0
Bank Sta=276.3,292.5
XS Rating Curve= 0 ,0
Exp/Cntr(USF)=0,0
Exp/Cntr=0.3,0.1

Type RM Length L Ch R = 1 ,16116   ,127.2,120.1,115.3
XS GIS Cut Line= 3
2160152.57988934 446176.812832232160081.81892458446202.326567619
 2159988.0950179446331.436324292
#Sta/Elev= 30
       0 3668.94     4.7 3668.38     8.9 3668.24    13.1 3668.31    19.4 3668.05
    34.4 3668.04    47.2 3667.16    50.6 3666.76    59.9 3666.35    71.8 3665.48
    75.6 3664.82    89.9 3659.66    93.6 3658.16    98.5 3656.56   103.5 3655.14
   112.1 3653.31   115.7 3652.53   118.3 3652.22     130 3652.07   141.4 3652.38
152.26433653.416   159.7 3653.43   172.9 3655.53   180.2 3656.31   187.5 3657.79
   197.4 3658.95   202.3 3659.78   221.6 3661.53     227 3661.65   234.8 3662.87
#Mann= 5 ,-1,0
       0      .1       0      70     .12       0   112.1    .045       0
152.2643     .12       0  165.22      .1       0
Bank Sta=112.1,152.2643
XS Rating Curve= 0 ,0
Exp/Cntr(USF)=0,0
Exp/Cntr=0.3,0.1

Type RM Length L Ch R = 1 ,15996   ,118.4,120.3,122.7
XS GIS Cut Line= 2
2159967.66521499446076.5024789972159909.27037896446311.506087407
#Sta/Elev= 30
       0 3656.43    21.3 3656.43    29.5 3656.28    37.8 3656.84    43.1 3656.49
    49.7 3656.44    62.5  3657.2    66.6  3656.8    82.7 3654.09    97.4 3651.29
   107.9 3649.79     112 3648.77   116.1 3647.38     119 3646.75   124.3 3645.77
   127.8  3645.6   144.2 3645.43   149.1 3645.54   157.3 3645.03   161.4 3645.04
   165.6 3645.31   173.8 3647.22   186.2 3649.19   198.5 3652.15   202.7 3652.86
   206.8 3653.15     210 3653.67   227.4 3656.97   235.6 3658.03   242.2 3658.68
#Mann= 5 ,-1,0
       0      .1       0     110     .12       0   127.8    .045       0
   144.2     .12       0     210      .1       0
Bank Sta=127.8,144.2
XS Rating Curve= 0 ,0
Exp/Cntr(USF)=0,0
Exp/Cntr=0.3,0.1

Type RM Length L Ch R = 1 ,15875   ,176.7,175.3,170.8
XS GIS Cut Line= 2
 2159863.7804237446065.4845621752159782.65647082446283.818163756
#Sta/Elev= 30
       0 3651.71    16.7 3650.99    25.3 3650.38    33.7 3650.28    38.1 3649.96
      43 3649.96    50.9  3650.4    55.5 3649.95    63.7 3647.82    72.2 3645.29
      85 3644.41    89.3 3643.42    97.8 3638.72   108.8 3634.57   117.7 3630.52
   122.4 3628.79   123.9  3628.4   130.1 3628.26   149.5 3628.89   153.3 3629.83
   164.3 3633.98   173.7 3636.28   178.9 3637.87   183.2 3639.68   187.4 3641.85
   191.7 3643.44     196 3644.18   204.8 3644.95   217.2 3647.14   232.9 3648.63
#Mann= 4 ,-1,0
       0      .1       0     120     .12       0   122.4    .045       0
   149.5     .12       0
Bank Sta=122.4,149.5
XS Rating Curve= 0 ,0
Exp/Cntr(USF)=0,0
Exp/Cntr=0.3,0.1

Type RM Length L Ch R = 1 ,15700   ,106.5,102.1,97.9
XS GIS Cut Line= 2
2159672.75315596446013.9641192512159639.74133443446248.103520162
#Sta/Elev= 30
       0 3644.14     7.3 3643.85    15.4 3643.15    23.4 3642.84    27.5 3642.37
    39.6 3643.37    40.7 3643.32    47.7 3642.65    55.8 3641.32    59.8 3639.35
    63.8 3635.96    67.9 3633.47      80 3631.22      84 3629.53    95.4 3623.03
    98.9  3621.3   100.2 3620.76   108.3 3619.29   112.3  3619.1   130.8 3619.19
   136.6 3619.42   144.6 3620.36   172.9  3622.9   176.9 3624.15     185 3625.43
   193.1  3626.5   205.2 3627.77   217.3  3629.9   225.4 3630.77   236.5 3632.65
#Mann= 3 ,-1,0
       0      .1       0   108.3    .045       0   136.6      .1       0
Bank Sta=108.3,136.6
XS Rating Curve= 0 ,0
Exp/Cntr(USF)=0,0
Exp/Cntr=0.3,0.1

Type RM Length L Ch R = 1 ,15598   ,119.8,123.8,128.1
XS GIS Cut Line= 3
2159563.17415567445998.8800750072159548.21938059446097.154311251
2159591.65944154446250.262722791
#Sta/Elev= 30
       0 3637.35     6.4 3637.97    18.5 3637.08    26.6 3637.68    34.7 3636.82
    46.8 3636.09      63 3636.19    71.1 3635.56    75.2 3634.32    79.2 3632.58
    87.3 3628.14    91.3  3626.3    99.4 3624.79   111.9 3616.77   120.2 3611.03
   125.3 3609.42   128.5 3608.78   132.7 3608.72   145.2 3609.16   153.5 3609.05
   157.7 3609.47   174.3 3611.15   182.6 3611.71   195.1 3616.27   207.5 3619.59
   215.9 3620.88   224.2 3621.66   228.3 3621.75     245 3624.19   258.6 3627.34
#Mann= 3 ,-1,0
       0      .1       0   125.3    .045       0   157.7      .1       0
Bank Sta=125.3,157.7
XS Rating Curve= 0 ,0
Exp/Cntr(USF)=0,0
Exp/Cntr=0.3,0.1

Type RM Length L Ch R = 1 ,15474   ,139.4,154.7,178.3
XS GIS Cut Line= 3
2159496.21881003445998.3820332482159436.12699308446113.558015734
2159460.16371986446291.830406016
#Sta/Elev= 30
       0 3633.28      11  3633.2    21.2 3632.39    52.8 3628.25    70.8 3626.32
    75.3  3625.2    79.9 3623.21    91.1 3619.93    93.4  3619.7   102.9 3620.51
   106.9 3619.37   129.9 3611.15   145.7  3608.3   158.1 3605.56   173.9 3601.34
     178 3600.81   193.6 3600.74   210.3 3601.01   213.4 3601.54   226.4 3606.08
   230.4 3607.97   242.5 3616.11   250.5 3621.06   254.6 3623.28   258.7 3624.95
   262.7 3626.05   278.9 3628.92   282.6 3629.97     295 3635.19   309.8 3640.75
#Mann= 3 ,-1,0
       0      .1       0   173.9    .045       0   213.4      .1       0
Bank Sta=173.9,213.4
XS Rating Curve= 0 ,0
Exp/Cntr(USF)=0,0
Exp/Cntr=0.3,0.1

Type RM Length L Ch R = 1 ,15319   ,160.3,168.5,184.2
XS GIS Cut Line= 2
2159432.36077238446004.3404968622159229.70394892 446223.88538894
#Sta/Elev= 30
       0 3627.19    17.5    3625    26.2 3622.96    35.7 3621.58    41.6 3619.59
    48.8 3615.64    51.7 3614.55    71.5 3609.04    82.8 3605.34    94.6 3602.61
   115.5 3599.55   120.9 3599.16   131.8 3598.98   153.6 3600.53   162.1 3600.35
   169.9 3600.68   175.3 3600.19   190.4  3596.6     196 3596.02   201.7 3596.32
   218.5 3596.15   224.4 3596.93   227.2 3599.36   235.2 3609.96   255.5 3627.12
   261.1 3632.24   266.8 3636.35   269.6 3637.68   273.3 3638.83   298.8 3644.77
#Mann= 3 ,-1,0
       0      .1       0   190.4    .045       0   224.4      .1       0
#XS Ineff= 2 , 0
          164.52 3611.55
Permanent Ineff=
       F       F
Bank Sta=190.4,224.4
XS Rating Curve= 0 ,0
Exp/Cntr(USF)=0,0
Exp/Cntr=0.3,0.1
