HEC-RAS study DOGWAYFK.prj: DOGWAYFK

--- DOGWAYFK.g01 (geometry) --- (continued)

Type RM Length L Ch R = 1 ,15151   ,158.5,141.5,122.1
XS GIS Cut Line= 3
2159367.87905582445952.1410120332159164.45459288446025.066762898
2159138.35485047446071.892771348
#Sta/Elev= 30
       0 3621.83    16.7 3617.92    28.7 3614.26    38.1 3609.26    42.2 3608.32
    50.7 3607.61    54.9 3605.79    63.4 3601.41    67.7 3599.92    76.2 3597.99
    81.9 3597.05    93.2 3593.94   103.8 3592.86   114.4 3592.68   123.6 3590.01
   127.2 3589.56   135.7 3589.49   150.7 3589.74   153.8 3590.19   161.2  3592.3
   169.7 3593.29   173.9 3593.16   182.4 3591.86   195.2 3591.75   200.8 3592.89
     207 3594.63   216.7 3598.05   225.4 3600.36   257.6 3602.97   269.7 3604.55
#Mann= 3 ,-1,0
       0      .1       0   123.6    .045       0   153.8      .1       0
#XS Ineff= 2 , 0
                          169.12         3598.63
Permanent Ineff=
       F       F
Bank Sta=123.6,153.8
XS Rating Curve= 0 ,0
Exp/Cntr(USF)=0,0
Exp/Cntr=0.3,0.1

Type RM Length L Ch R = 1 ,15009   ,198.4,195.3,190.9
XS GIS Cut Line= 3
2159156.79061192445825.0631404482159145.78667141445930.823235377
2159128.29453299446069.452750177
#Sta/Elev= 30
       0 3622.94     4.3 3621.62    12.2 3617.41    16.2 3615.63    35.3 3604.34
    48.4 3598.36    52.4 3595.58    58.9    3590    64.5  3585.7    68.5 3584.38
    77.2 3584.31    80.5 3584.31    84.6 3585.23    92.6 3588.77    96.6  3589.8
   100.7  3590.1   104.7  3590.8   108.7 3590.85   112.7 3590.33   120.8 3588.17
   127.8 3587.56   132.9  3587.5   161.1  3588.8   169.2 3589.56   177.2 3589.85
   192.2 3591.06   197.4 3592.27   206.5 3595.26   221.6 3598.96   246.1  3603.7
#Mann= 3 ,-1,0
       0      .1       0    64.5    .045       0    84.6      .1       0
#XS Ineff= 2 , 0
                          107.84         3599.16
Permanent Ineff=
       F       F
Bank Sta=64.5,84.6
XS Rating Curve= 0 ,0
Exp/Cntr(USF)=0,0
Exp/Cntr=0.3,0.1

Type RM Length L Ch R = 1 ,14814   ,167,165.4,163
XS GIS Cut Line= 2
2158949.75511278445844.914009229 2158996.2333323446104.772121978
#Sta/Elev= 30
       0 3608.59     4.3 3607.79    12.5 3607.05    16.5 3606.02    28.7 3600.63
    36.8 3596.55      49 3588.24    53.1 3586.96    61.2  3585.8    69.3 3581.16
    73.4  3580.1    85.6 3579.77   101.9 3579.84   118.1 3577.94   126.2 3577.56
   134.4 3577.89   146.6 3581.91   150.6 3582.69   166.9 3581.76   195.5 3581.85
   203.4 3582.66   211.6 3584.94   219.7 3586.55   223.8 3587.65   227.8 3589.59
   239.8 3598.27   244.1 3601.07   252.2  3605.6   256.3 3607.46     264 3611.63
#Mann= 3 ,-1,0
       0      .1       0   118.1    .045       0   134.4      .1       0
Bank Sta=118.1,134.4
XS Rating Curve= 0 ,0
Exp/Cntr(USF)=0,0
Exp/Cntr=0.3,0.1

Type RM Length L Ch R = 1 ,14649   ,192.3,205.6,214.5
XS GIS Cut Line= 2
2158808.16750596 445894.222883872158855.23942924446126.577909406
#Sta/Elev= 30
       0 3583.21     7.1 3582.43    23.4 3581.81    27.5 3581.09    35.7  3578.1
    39.7 3577.57    43.8 3578.31      52 3578.46    56.8  3577.6    64.2 3577.36
    72.4 3576.26    77.2 3576.63    97.5 3573.38   100.9 3572.97   109.1 3572.68
   113.2 3572.78   125.5 3575.16   131.5 3574.94   138.3 3573.75   141.8 3573.03
   145.9 3572.84     154 3572.98   157.3 3573.63   178.5 3578.31   185.8 3580.43
   190.8 3582.27   203.4 3585.47   211.2 3587.78   219.3 3591.99   237.1 3602.22
#Mann= 3 ,-1,0
       0      .1       0   138.3    .045       0   157.3      .1       0
Bank Sta=138.3,157.3
XS Rating Curve= 0 ,0
Exp/Cntr(USF)=0,0
Exp/Cntr=0.3,0.1

Type RM Length L Ch R = 1 ,14443   ,180.8,199.5,209.9
XS GIS Cut Line= 2
2158725.04049252445858.1677937012158608.86297975446041.447835395
#Sta/Elev= 30
       0 3579.43     3.6 3579.01      13 3576.57    22.5 3574.94    31.5  3572.5
    34.7 3571.97    41.5 3569.77    50.9 3567.83    55.7 3567.22    60.4 3567.51
    66.6 3568.59    74.6 3569.39    93.5 3569.29     103 3570.41   113.7 3570.98
   117.2 3570.81   121.7 3570.23   131.4 3567.67   136.1 3567.22   144.8 3567.21
   159.9 3567.56   169.3  3570.4   176.7 3577.11   178.8 3579.43   185.4 3588.35
   188.3 3591.56   194.1 3595.01   197.7 3597.44   210.8 3602.06     217 3605.06
#Mann= 3 ,-1,0
       0      .1       0   131.4    .045       0   159.9      .1       0
#XS Ineff= 2 , 0
          113.67 3578.14
Permanent Ineff=
       F       F
Bank Sta=131.4,159.9
XS Rating Curve= 0 ,0
Exp/Cntr(USF)=0,0
Exp/Cntr=0.3,0.1

Type RM Length L Ch R = 1 ,14244   ,208.3,196.9,184.8
XS GIS Cut Line= 2
2158715.02518969445799.0775070352158478.66404303445845.147900029
#Sta/Elev= 30
       0  3588.7     4.2 3587.98    15.1 3584.47    23.3 3582.33    31.5 3579.06
    38.3 3578.29    51.8  3577.5      60 3576.21    68.1 3575.54    72.2 3574.46
    86.1 3566.26    92.6 3563.42    96.6 3563.13   108.9 3559.73   112.9 3559.11
   121.1 3559.36   129.2 3558.52   137.2 3558.14   145.5 3558.35   149.6 3559.02
   154.3  3560.4   178.2 3568.46   190.4 3570.85   194.4 3571.24   198.6 3571.03
   202.6 3571.25   220.1 3573.94   225.9 3575.17   239.3 3579.27   240.8 3579.48
#Mann= 3 ,-1,0
       0      .1       0   129.2    .045       0   145.5      .1       0
Bank Sta=129.2,145.5
XS Rating Curve= 0 ,0
Exp/Cntr(USF)=0,0
Exp/Cntr=0.3,0.1

Type RM Length L Ch R = 1 ,14047   ,217.8,199.4,185
XS GIS Cut Line= 2
2158551.77575365445605.7821625162158414.56610495445759.016295735
#Sta/Elev= 30
       0 3584.31    13.5 3575.52      22 3569.49    35.4 3559.08    41.4 3555.08
    52.9    3551    55.9 3550.65    63.6 3550.28    85.1 3550.51    89.3 3550.84
    90.5 3551.11    95.8 3553.05   101.3  3553.7   113.3 3554.41   121.1 3556.16
   123.9 3556.58   125.3 3556.67   132.4  3556.4   137.3 3555.74   155.3  3554.9
   160.3 3555.12   167.3 3556.08   177.8 3556.55   181.7 3557.19   187.1 3558.77
   191.9 3559.93   197.6 3560.73   200.4 3561.32   203.3 3562.21   205.7 3563.19
#Mann= 3 ,-1,0
       0     .06       0    52.9    .045       0    89.3      .1       0
Bank Sta=52.9,89.3
XS Rating Curve= 0 ,0
Exp/Cntr(USF)=0,0
Exp/Cntr=0.3,0.1

Type RM Length L Ch R = 1 ,13847   ,182.1,187.4,187.2
XS GIS Cut Line= 2
2158319.42072811445517.6474976572158326.43144009445728.970387261
#Sta/Elev= 30
       0 3580.57     7.5 3579.16    11.5 3577.96    15.5 3575.73    40.1 3554.67
    47.6 3549.15    51.6  3546.5    55.6 3543.41    59.6 3540.92    63.6 3540.29
    83.6 3540.02    87.6 3540.23    89.4 3540.77    91.6 3541.42    99.6 3545.52
   103.6 3546.47   107.6  3546.7   115.6 3546.46   135.6 3546.97   147.6 3546.32
   155.2 3546.83   163.6 3546.89   167.6 3547.11   176.7 3548.31   179.6 3548.81
   183.6 3549.83   189.2 3551.87   199.6  3556.2   207.6 3560.16   211.4 3561.71
#Mann= 3 ,-1,0
       0     .06       0    59.6    .045       0    89.4      .1       0
Bank Sta=59.6,89.4
XS Rating Curve= 0 ,0
Exp/Cntr(USF)=0,0
Exp/Cntr=0.3,0.1

Type RM Length L Ch R = 1 ,13660   ,208.8,213.8,213.7
XS GIS Cut Line= 2
2158149.16058009445530.6673913292158130.13150472445722.961205566
#Sta/Elev= 30
       0 3556.48     2.5 3554.18     6.5 3550.91    10.6  3548.5    14.6 3546.78
    22.6 3543.82    30.7 3542.02    41.9 3540.77    46.7 3539.87    54.8 3538.86
    58.1 3537.87    66.8 3534.38    70.9 3533.19    74.9 3532.85    87.3 3532.53
      95 3532.06      99 3532.21     103 3532.95     107 3533.74   111.1 3535.81
   119.1 3540.41   123.1 3541.29   131.1 3541.84   139.2  3545.5   143.2  3546.1
   151.2 3546.74   159.3 3548.19   171.2 3549.03   189.1 3552.76   193.2 3553.94
#Mann= 4 ,-1,0
       0     .06       0      60      .1       0    70.9    .045       0
     103      .1       0
Bank Sta=70.9,103
XS Rating Curve= 0 ,0
Exp/Cntr(USF)=0,0
Exp/Cntr=0.3,0.1

Type RM Length L Ch R = 1 ,13446   ,198.5,204,210.3
XS GIS Cut Line= 2
2157956.86676585445484.5969983352157921.81320597445641.837252685
#Sta/Elev= 30
       0 3551.15     8.8 3546.54    12.9 3544.57      21 3541.18    25.2 3539.08
    29.3 3537.62    33.4  3536.3    37.5 3534.41    39.9  3533.1    41.6 3532.27
    49.8 3530.27    54.7 3528.74    70.3 3524.62    74.4 3524.16    81.5 3523.57
    90.8 3523.31    94.9 3523.41    98.2 3523.84      99 3523.98   103.1 3525.13
   107.1 3527.16   111.7 3529.74   115.3 3531.66   119.4 3532.89   127.6 3533.65
   135.8 3535.48     144 3537.05   148.5 3537.57   156.3 3539.01   161.1 3539.61
#Mann= 4 ,-1,0
       0     .06       0      10      .1       0    74.4    .045       0
    98.2      .1       0
Bank Sta=74.4,98.2
XS Rating Curve= 0 ,0
Exp/Cntr(USF)=0,0
Exp/Cntr=0.3,0.1

Type RM Length L Ch R = 1 ,13242   ,203.6,202.7,200.7
XS GIS Cut Line= 2
2157830.67395026445387.4485609342157716.49949806445538.679633589
#Sta/Elev= 30
       0 3553.81     4.1 3552.13    11.6 3550.11    14.4 3548.96    24.1 3543.56
    30.7 3540.61    34.4 3538.53    37.3 3536.56    57.3 3519.71    60.1 3517.81
    62.3 3516.92    71.6 3515.97    80.1 3514.51    85.8 3513.89    92.4 3513.95
    97.1 3514.41     103 3516.47   108.7 3520.39   112.4 3523.51   114.4 3524.66
   117.4 3525.91   123.6 3527.07   128.7 3527.62   137.5 3527.13   147.5 3526.53
   160.1 3525.02   165.8 3524.65   168.7 3524.83   177.2 3526.25   189.5 3527.48
#Mann= 3 ,-1,0
       0      .1       0    80.1    .045       0    97.1      .1       0
Bank Sta=80.1,97.1
XS Rating Curve= 0 ,0
Exp/Cntr(USF)=0,0
Exp/Cntr=0.3,0.1

Type RM Length L Ch R = 1 ,13039   ,214,213.3,211.2
XS GIS Cut Line= 2
2157644.38931772445291.3016538162157549.24394088445488.603119465
#Sta/Elev= 30
       0 3549.97     4.6    3549      11 3547.17    18.9 3543.71    28.7 3536.43
    33.2 3533.54    42.1 3526.84    55.4 3518.48    59.8 3515.85    61.5 3515.12
    64.3 3514.08    73.1 3514.08    79.5 3513.14    83.4  3512.3    91.4 3509.63
    99.8 3507.23   104.2 3506.46     111 3505.54   117.5 3505.26   139.7 3505.53
   147.8 3506.61   153.1 3507.82     162 3511.99   166.3 3512.87   184.2 3513.17
   188.6 3513.46   192.3 3514.32   201.9 3517.67   212.3 3520.51     219 3523.25
#Mann= 4 ,-1,0
       0     .06       0      40      .1       0   104.2    .045       0
   147.8      .1       0
Bank Sta=104.2,147.8
XS Rating Curve= 0 ,0
Exp/Cntr(USF)=0,0
Exp/Cntr=0.3,0.1

Type RM Length L Ch R = 1 ,12826   ,193.3,196.2,198.4
XS GIS Cut Line= 2
2157454.09856405445191.1486255682157350.94094495445444.535787036
#Sta/Elev= 30
       0 3542.02     6.5 3540.63    10.8 3538.87    36.7 3523.95    49.1 3517.61
      54  3514.5    58.1 3512.73    62.7 3511.98    75.6  3513.5    79.8  3513.5
    84.2 3512.98   101.5 3505.21   105.8 3502.88   110.2 3501.88   123.1 3499.99
   138.6  3495.2   140.4 3494.81     149 3494.68   157.7 3494.79   160.63495.395
   166.3 3497.18   170.6 3499.67   174.9 3503.35   179.3 3505.46   187.2 3506.59
   196.5 3506.91   213.8 3510.46   235.4 3513.17   261.3 3519.75   273.6 3521.62
#Mann= 3 ,-1,0
       0      .1       0   138.6    .045       0   160.6      .1       0
Bank Sta=138.6,160.6
XS Rating Curve= 0 ,0
Exp/Cntr(USF)=0,0
Exp/Cntr=0.3,0.1

Type RM Length L Ch R = 1 ,12630   ,184.4,182.3,183
XS GIS Cut Line= 2
2157297.31346184445119.5456566682157178.13135822445320.853243447
#Sta/Elev= 30
       0 3535.89     6.5 3532.78    15.8 3529.06    25.8 3524.67    29.8 3522.67
    33.6 3520.18    41.5 3514.02    45.8 3511.11    63.3 3500.38    72.1 3495.37
      75 3494.23    80.9 3493.32    86.7 3493.56    98.4 3492.15   104.3  3490.1
   108.8 3489.08   113.5 3488.85   122.8 3488.92   136.3  3489.5   139.3 3490.05
     146 3491.55   159.7 3492.46   164.6 3493.26   168.5 3494.89   173.9 3498.26
   178.5 3499.57   200.6 3500.96   209.3 3502.01   222.1 3504.21   233.9  3505.1
#Mann= 3 ,-1,0
       0      .1       0   104.3    .045       0   139.3      .1       0
Bank Sta=104.3,139.3
XS Rating Curve= 0 ,0
Exp/Cntr(USF)=0,0
Exp/Cntr=0.3,0.1

Type RM Length L Ch R = 1 ,12448   ,194.3,197.6,199.7
XS GIS Cut Line= 2
2157158.64713071445015.8808261342157010.42064891445247.234321387
#Sta/Elev= 30
       0 3526.41     1.5  3525.9      11 3523.97    17.2    3522    34.6 3517.85
    40.4 3515.95    49.1 3514.06    53.8 3513.42    63.3 3511.06    93.6    3501
    98.3 3498.66   101.3  3496.7   112.8 3490.29   118.5 3487.85   124.3 3486.67
   127.2 3486.34   134.6 3485.94   144.1 3484.68   158.3 3483.73   164.9 3483.45
   173.6 3483.58   177.3 3483.93   196.3 3491.26   201.1 3492.47   220.1 3495.23
   229.6 3496.34   243.8 3497.11   256.7  3498.5   264.1 3499.55   274.8 3501.69
#Mann= 3 ,-1,0
       0      .1       0   158.3    .045       0   177.3      .1       0
Bank Sta=158.3,177.3
XS Rating Curve= 0 ,0
Exp/Cntr(USF)=0,0
Exp/Cntr=0.3,0.1

Type RM Length L Ch R = 1 ,12250   ,202.3,202.2,201.1
XS GIS Cut Line= 2
2157010.42064891444936.7599338182156850.17580371445105.017021275
#Sta/Elev= 30
       0 3502.19     6.1 3498.41    13.2 3493.64    20.7 3489.24    22.7 3488.32
    30.2 3485.61    33.7 3484.83    47.2 3483.66    69.8 3482.68    72.9 3482.16
    83.9 3478.27    90.23476.334   100.9 3475.74   116.6 3475.48   122.1 3476.01
   125.1 3476.18   130.9 3477.14   142.5 3481.48   146.2 3482.17   151.8 3482.68
   159.9 3482.95   166.3 3483.56   182.9 3483.19   194.7 3483.64   199.9 3484.32
     205 3485.82   210.5 3488.13     216 3489.33   221.5 3489.82   232.4 3489.69
#Mann= 3 ,-1,0
       0      .1       0    90.2    .045       0   122.1      .1       0
Bank Sta=90.2,122.1
XS Rating Curve= 0 ,0
Exp/Cntr(USF)=0,0
Exp/Cntr=0.3,0.1

Type RM Length L Ch R = 1 ,12048   ,200.3,205.1,209.5
XS GIS Cut Line= 2
 2156845.1681523444814.5732393552156709.96156416444966.805842292
#Sta/Elev= 30
       0 3476.79     5.4 3476.28    24.9 3475.15      28 3475.12    35.6  3475.4
    40.9 3475.06    51.6 3474.72      57 3473.55    67.7 3470.66      73 3469.46
    79.8 3469.19    83.7 3469.17    89.1 3469.22    91.8 3469.51    94.4 3470.06
    99.8 3472.61   105.1 3473.58   113.1 3473.71   115.9 3473.94     128 3477.29
   131.9 3477.98   141.4 3479.28   147.9 3479.29   153.3 3479.08   164.1 3478.34
   170.2 3478.71   178.2 3479.45   192.4 3480.29   195.2  3480.6   203.6  3480.8
#Mann= 3 ,-1,0
       0      .1       0      73    .045       0    91.8      .1       0
Bank Sta=73,91.8
XS Rating Curve= 0 ,0
Exp/Cntr(USF)=0,0
Exp/Cntr=0.3,0.1

Type RM Length L Ch R = 1 ,11843   ,182.8,186.7,191.4
XS GIS Cut Line= 3
  2156759.036548444664.3436969822156544.70906755444809.565587942
2156460.58052382444930.750752123
#Sta/Elev= 30
       0 3484.78    22.9 3479.13    31.5 3474.87    42.1 3470.65    56.6 3468.19
    61.4 3467.67    71.1 3468.23    80.8 3467.72    94.8 3464.92   109.8 3466.32
   117.9 3466.09   124.2 3465.44     137 3462.89   151.2 3462.23   169.7 3462.84
   178.4 3466.18     187  3471.6   189.9 3471.89   222.5 3471.87   243.9 3468.45
   266.8  3466.5   287.9 3466.37   297.4 3466.82   308.9 3468.43   330.9 3474.51
     344 3476.38   360.7 3480.22   375.3 3486.43   382.6 3488.65   406.4 3497.88
#Mann= 3 ,-1,0
       0      .1       0     137    .045       0   169.7      .1       0
#XS Ineff= 2 , 0
       0   109.8    3468               0
Permanent Ineff=
       F       F
Bank Sta=137,169.7
XS Rating Curve= 0 ,0
Exp/Cntr(USF)=0,0
Exp/Cntr=0.3,0.1

Type RM Length L Ch R = 1 ,11656   ,228.7,219.6,212.5
XS GIS Cut Line= 3
2156699.94626134444533.1432299772156506.65091682444601.247289186
2156301.33720891444898.701783083
#Sta/Elev= 30
       0 3489.21    65.7 3478.39    80.3 3473.45    96.4 3465.54   114.3 3458.04
   122.7 3457.34   144.83458.174   173.6 3463.63   197.4 3463.05   209.3 3463.87
   238.9 3461.14   286.8 3460.64   321.5 3458.63   336.1  3460.5   355.5 3461.68
   365.2 3460.53   376.3 3460.71   394.4 3459.59   399.3 3461.54   418.7 3471.81
   438.2 3476.03   462.8 3483.62   474.1 3486.44   491.6 3492.84   505.7 3495.78
   511.5 3498.27   525.6 3502.72   540.2 3506.16   557.5 3512.95   566.4 3515.49
#Mann= 3 ,-1,0
       0      .1       0   114.3    .045       0   144.8      .1       0
#XS Ineff= 2 , 0
                          203.16         3474.13
Permanent Ineff=
       F       F
Bank Sta=114.3,144.8
XS Rating Curve= 0 ,0
Exp/Cntr(USF)=0,0
Exp/Cntr=0.3,0.1

Type RM Length L Ch R = 1 ,11436   ,191.8,187.6,181.9
XS GIS Cut Line= 3
2156545.71059783444305.7958558542156355.41984416444496.086609526
2156086.00819817444761.492134383
#Sta/Elev= 30
       0 3478.13    36.1 3466.53      50 3460.62    82.7 3457.91   109.7 3457.52
   127.9 3452.67   133.6  3451.6   147.7 3452.86   157.5 3454.81   171.9 3454.81
     193 3458.03   215.6 3459.26   259.3  3458.7   304.9 3459.97   331.6 3459.13
   346.7 3456.05   365.5 3454.05   385.3 3453.23   405.1 3451.17     414 3452.39
   425.3 3450.37     456 3450.84   470.2 3451.53   475.9 3452.73   487.3 3457.02
   504.1 3465.63   521.5  3472.4     572 3489.11     589 3493.69   647.3 3514.01
#Mann= 3 ,-1,0
       0      .1       0   127.9    .045       0   147.7      .1       0
#XS Ineff= 2 , 0
                          216.39         3465.74
Permanent Ineff=
       F       F
Bank Sta=127.9,147.7
XS Rating Curve= 0 ,0
Exp/Cntr(USF)=0,0
Exp/Cntr=0.3,0.1

Type RM Length L Ch R = 1 ,11249   ,161.8,156.9,149.3
XS GIS Cut Line= 3
2156358.42443501444172.5923282842156246.25304337444405.948884102
2156003.88271501 444679.36665122
#Sta/Elev= 30
       0 3462.92    32.1 3454.01    49.5 3453.24    62.8 3453.72    76.1 3451.17
     116 3447.84   133.8 3447.27     137 3447.94   147.1 3451.36   169.3 3454.08
   187.1 3453.57   208.9 3451.41   218.1 3451.56   231.4 3454.02   235.9 3454.07
   285.3 3450.75   352.5 3452.98     359  3451.7   370.1  3447.6     376 3446.76
   382.7  3446.7   394.7 3448.79   449.7 3446.27     477 3447.59   519.8  3462.9
   535.8 3467.13   575.6  3482.4   587.7 3488.04     597 3493.41   624.3 3505.81
#Mann= 3 ,-1,0
       0      .1       0     116    .045       0     137      .1       0
#XS Ineff= 2 , 0
                          179.15         3468.27
Permanent Ineff=
       F       F
Bank Sta=116,137
XS Rating Curve= 0 ,0
Exp/Cntr(USF)=0,0
Exp/Cntr=0.3,0.1

Type RM Length L Ch R = 1 ,11092   ,190.5,198.6,203.5
XS GIS Cut Line= 3
2156158.11837851444186.6137522392156147.10154541444415.964186927
2155940.78630722444649.320742745
#Sta/Elev= 30
       0 3456.21    30.6 3455.32    42.6 3454.13    62.6 3449.26    70.6 3445.59
    78.7  3443.6    98.7 3442.63   106.7 3443.61   158.7 3446.74   174.8 3446.48
   198.8 3452.35   222.8 3453.73   231.2 3452.67   247.3  3452.4   263.7 3448.57
   288.4  3445.6   306.5 3445.73   327.3 3444.11     338 3445.84   343.4 3445.31
   351.6 3443.31   360.1 3442.55   374.2 3444.11   380.7 3445.48   403.1 3452.99
   425.2 3461.28   436.6 3464.41   475.6 3480.28   499.7 3491.87   541.1 3505.73
#Mann= 3 ,-1,0
       0      .1       0    78.7    .045       0   106.7      .1       0
#XS Ineff= 2 , 0
                          207.91         3471.79
Permanent Ineff=
       F       F
Bank Sta=78.7,106.7
XS Rating Curve= 0 ,0
Exp/Cntr(USF)=0,0
Exp/Cntr=0.3,0.1

Type RM Length L Ch R = 1 ,10893   ,245.8,251.5,251.5
XS GIS Cut Line= 2
2156032.81311254444129.1906787052155821.43627988 444457.49479264
#Sta/Elev= 30
       0 3444.69     9.5 3444.29    33.3 3444.46    52.3 3445.36    57.1 3444.95
    71.3 3444.91    85.6 3442.84    90.2 3441.23    95.1 3438.13    99.9 3437.15
   116.2 3437.16   137.9 3439.28   161.7 3439.05   171.3 3437.83     195 3437.29
   218.8 3435.95   249.3 3435.42   266.7 3434.33   278.3 3435.41   295.6 3439.26
   304.5 3439.46   310.1 3441.08   318.9 3444.37   326.3  3446.1   337.8 3448.02
   355.9 3452.55   362.2 3454.81   370.6 3458.75     378 3461.71   390.5 3465.38
#Mann= 3 ,-1,0
       0      .1       0    99.9    .045       0   116.2      .1       0
#XS Ineff= 2 , 0
                             268         3454.91
Permanent Ineff=
       F       F
Bank Sta=99.9,116.2
XS Rating Curve= 0 ,0
Exp/Cntr(USF)=0,0
Exp/Cntr=0.3,0.1

Type RM Length L Ch R = 1 ,10642   ,188.2,189.3,189.1
XS GIS Cut Line= 2
 2155827.6133853444051.4071641042155512.13134631444442.003974271
#Sta/Elev= 30
       0 3438.74     9.4 3439.38    24.6 3439.21    29.3 3438.14    37.8 3433.69
    48.6  3432.4    53.7 3431.01    88.2 3430.06   111.8 3429.78   120.1 3430.21
   139.2 3430.76   154.5 3429.88   185.7 3430.82   197.7 3433.18   208.5 3434.07
   231.3 3432.12   243.9 3432.94   259.4 3431.69   271.1  3432.9   296.7 3440.82
   315.9 3450.08   325.1 3452.73   364.9 3469.07   377.6 3473.49   393.1 3478.64
   418.8  3486.1   444.5 3491.15     473 3498.76   495.7 3507.04   502.1 3510.48
#Mann= 3 ,-1,0
       0      .1       0    88.2    .045       0   120.1      .1       0
#XS Ineff= 2 , 0
                          207.91         3450.77
Permanent Ineff=
       F       F
Bank Sta=88.2,120.1
XS Rating Curve= 0 ,0
Exp/Cntr(USF)=0,0
Exp/Cntr=0.3,0.1

Type RM Length L Ch R = 1 ,10453   ,209,206.9,204.6
XS GIS Cut Line= 4
2155764.40932444443928.0613808412155660.10804506443958.474315013
2155534.28747877444130.5325193742155484.13041744444313.376306063
#Sta/Elev= 30
       0 3433.01    17.2 3433.81    37.7 3433.07    87.7  3433.2     104 3432.13
   116.3 3432.55   139.2 3430.55148.71913426.391161.91853426.591   171.5 3428.64
   189.8 3428.97   211.1 3427.08     226 3427.63   239.3  3426.9   256.5 3424.66
   276.5 3430.01   296.6    3431   328.7 3431.13     381  3428.2   411.6 3428.41
   423.3 3429.53   428.2 3431.87   436.3 3438.73     449 3446.17   459.1 3455.44
   469.7 3461.28     478 3464.69   486.3 3466.69   494.6 3468.33   511.4 3470.25
#Mann= 3 ,-1,0
       0      .1       0148.7191    .045       0161.9185      .1       0
#XS Ineff= 2 , 0
                          300.85         3443.06
Permanent Ineff=
       F       F
Bank Sta=148.7191,161.9185
XS Rating Curve= 0 ,0
Exp/Cntr(USF)=0,0
Exp/Cntr=0.3,0.1

Type RM Length L Ch R = 1 ,10246   ,193.3,192,189.9
XS GIS Cut Line= 3
2155697.99007189443725.1558228242155504.17146255443800.666493513
2155298.80539615 444247.70709947
#Sta/Elev= 30
       0 3438.89    36.3 3437.47    87.8 3432.45   100.7 3433.66   117.9 3431.29
   165.2 3429.88   208.6 3426.45   248.2 3426.64   261.4  3423.8   287.8  3424.3
326.14093419.999   336.2 3419.69341.24093419.979   362.6 3425.19   384.6 3424.84
   411.1  3425.9   437.5 3425.28   450.7 3424.01   499.1 3424.03   529.9 3421.01
   542.9 3421.13   562.5 3424.24   591.3  3424.1   604.7 3422.05   612.6  3422.2
   622.4 3423.37   626.8 3424.88   657.6 3438.09     684 3445.08     700 3447.62
#Mann= 5 ,-1,0
       0      .1       0  228.01     .12       0  318.01      .1       0
326.1409    .045       0341.2409      .1       0
#XS Ineff= 2 , 0
          282.37 3427.65  434.99         3433.76
Permanent Ineff=
       F       F
Bank Sta=326.1409,341.2409
XS Rating Curve= 0 ,0
Exp/Cntr(USF)=0,0
Exp/Cntr=0.3,0.1

Type RM Length L Ch R = 1 ,10054   ,222.1,212.7,198.1
XS GIS Cut Line= 3
2155299.80692643443762.9664427492155189.63859535444115.505102182
2155258.74418485 444267.73770512
#Sta/Elev= 30
       0 3427.46    23.3 3426.38      40 3426.49    46.2 3424.99    65.8 3417.35
    73.6 3416.79    89.3 3417.32   102.9 3419.76   111.3 3422.09   132.2  3420.2
   186.7 3418.16   195.1 3418.45   203.5 3416.99   220.2 3417.49   232.8 3416.26
   249.6 3418.22   279.3 3419.31   314.4 3416.49   317.6 3416.78   329.2 3419.53
   337.6 3419.66   354.3    3421   369.5 3420.15   397.5 3421.13   415.1 3420.93
   428.3 3419.91     436 3420.18   445.9 3421.88   502.4 3438.73   536.5  3443.6
#Mann= 3 ,-1,0
       0      .1       0    65.8    .045       0    89.3      .1       0
#XS Ineff= 2 , 0
                          143.32         3430.26
Permanent Ineff=
       F       F
Bank Sta=65.8,89.3
XS Rating Curve= 0 ,0
Exp/Cntr(USF)=0,0
Exp/Cntr=0.3,0.1

Type RM Length L Ch R = 1 ,9841    ,207.9,211.2,214
XS GIS Cut Line= 4
2155025.38762903443758.9603216192155139.56208123443874.136304104
2155166.60339886444117.5081627472155212.67379185 444271.74382625
#Sta/Elev= 30
       0 3444.51      20 3442.45    42.6 3426.65    51.6 3421.45    57.3 3418.59
    70.7 3415.08    85.6 3415.22   130.8 3418.05   151.7 3417.44   172.7 3418.13
   241.7 3417.61   249.8 3416.36   261.8 3412.29     294 3413.94   322.2 3411.57
   330.2 3412.27   338.3 3415.71     343 3416.83   354.4 3418.39   366.5 3419.06
   382.8 3418.48   414.5 3419.34   440.1 3421.15   465.9 3418.91   477.7 3419.19
   485.2 3420.21   502.7 3424.69   538.3 3435.38   555.9 3439.03     568 3440.15
#Mann= 3 ,-1,0
       0      .1       0    70.7    .045       0    85.6      .1       0
#XS Ineff= 2 , 0
                          220.06         3431.05
Permanent Ineff=
       F       F
Bank Sta=70.7,85.6
XS Rating Curve= 0 ,0
Exp/Cntr(USF)=0,0
Exp/Cntr=0.3,0.1

Type RM Length L Ch R = 1 ,9630    ,184.8,184.7,185
XS GIS Cut Line= 3
2154967.14242018443949.0754598142155147.30990178444070.090209356
2155167.17799499444243.032929785
#Sta/Elev= 30
       0 3418.52    20.5 3413.77    29.6 3412.29    36.1 3411.99    54.2  3412.7
    68.7 3409.51    73.5 3408.78      88 3408.46   102.4 3408.59   107.8 3409.42
   126.5 3413.43   145.8 3414.31   155.4 3413.38   160.3 3411.92   174.7  3409.2
   179.5 3409.09   193.9 3411.09   201.1 3413.38   208.2  3417.1   215.4 3418.39
   244.3 3417.49   256.4 3418.72   276.5 3419.03   304.7 3418.01   316.8 3419.67
   320.8 3419.62   328.9 3417.84   340.9 3417.45   361.1 3419.64   391.1 3428.52
#Mann= 3 ,-1,0
       0      .1       0    68.7    .045       0   107.8      .1       0
#XS Ineff= 2 , 0
                          147.15         3421.73
Permanent Ineff=
       F       F
Bank Sta=68.7,107.8
XS Rating Curve= 0 ,0
Exp/Cntr(USF)=0,0
Exp/Cntr=0.3,0.1

Type RM Length L Ch R = 1 ,9445    ,181.9,182.4,182.7
XS GIS Cut Line= 2
2154840.10452677444040.3903309962155046.41976496444245.704038905
#Sta/Elev= 30
       0 3413.07     6.8 3410.94    22.7 3406.97      34  3405.7    45.9 3403.95
    50.9 3404.12    74.1 3406.25    80.5 3406.21    91.8 3404.63      96    3405
   105.3 3406.49   125.1    3407   133.5 3406.69   137.2 3406.85   146.8 3407.89
   159.9 3406.32   178.8 3403.24   186.3    3403   190.1 3403.26     192 3403.52
   195.8 3404.95   205.3  3407.9   209.9 3409.64   224.1    3413   233.6 3415.75
   243.9  3416.7   246.7 3416.68   267.6 3415.37   286.3 3415.53   291.1  3415.3
#Mann= 3 ,-1,0
       0      .1       0   178.8    .045       0   190.1      .1       0
Bank Sta=178.8,190.1
XS Rating Curve= 0 ,0
Exp/Cntr(USF)=0,0
Exp/Cntr=0.3,0.1

Type RM Length L Ch R = 1 ,9263    ,215,216.7,217.4
XS GIS Cut Line= 3
2154742.95608937444155.5663134822154788.02495208444244.702508623
2154900.19634372444356.873900261
#Sta/Elev= 30
       0 3406.76    15.3    3407    19.7 3406.77    33.2  3403.4    51.1 3401.12
    60.1 3400.82    70.6 3401.32    79.5 3402.11    85.5  3403.2    94.4 3404.22
   100.1 3404.47   106.2    3404   111.6 3402.98   114.5 3402.81   134.5 3402.43
   151.5 3402.85   156.9 3402.33   168.2 3399.85   173.6 3399.21   179.5 3399.04
   199.3 3399.25   202.4 3399.85   210.6 3404.49   213.2 3405.66   224.5 3406.46
   230.7 3408.39   236.1 3408.47   238.9 3408.18   247.2 3406.15   258.5 3406.67
#Mann= 3 ,-1,0
       0      .1       0   173.6    .045       0   199.3      .1       0
Bank Sta=173.6,199.3
XS Rating Curve= 0 ,0
Exp/Cntr(USF)=0,0
Exp/Cntr=0.3,0.1

Type RM Length L Ch R = 1 ,9046    ,200.4,198.1,194.4
XS GIS Cut Line= 2
2154471.54138282444193.6244642162154775.00505841444548.166184215
#Sta/Elev= 30
       0 3421.23    14.3  3409.9    19.4  3406.4    25.7 3402.64    31.3 3400.64
    62.6 3401.13   102.3 3399.47     125 3400.88   148.6 3400.43   154.8 3399.89
   161.8 3397.22   167.9 3396.01     204 3397.98   218.6 3399.52   227.1 3398.25
   252.6 3398.14   273.2  3396.4   283.7 3396.94   302.4 3396.53   320.8  3394.5
   331.1 3393.85   345.5 3393.91   349.1 3394.53   362.7 3400.26   377.4 3402.13
   380.3    3403   404.8 3417.14   420.6 3422.91   457.5 3433.99   466.7 3435.88
#Mann= 4 ,-1,0
       0     .12       0      20      .1       0   320.8    .045       0
   349.1      .1       0
#XS Ineff= 1 ,-1
  218.89  254.99 3406.57
Permanent Ineff=
       F
Bank Sta=320.8,349.1
XS Rating Curve= 0 ,0
Exp/Cntr(USF)=0,0
Exp/Cntr=0.3,0.1

Type RM Length L Ch R = 1 ,8848    ,214.5,211.3,208.7
XS GIS Cut Line= 2
2154321.31184044 444372.898384782154669.84437875444682.371242067
#Sta/Elev= 30
       0 3417.25    10.7 3413.79    19.9 3409.39    57.3 3396.41    62.7 3395.39
    73.1 3395.21    87.2 3392.59    94.8 3392.44   105.5  3393.8   163.1  3396.2
   203.4 3394.42   217.6 3392.13   229.4 3395.06   255.2 3394.21   260.1 3393.75
   269.5 3391.03   277.1 3390.56   295.6 3391.09   316.7 3393.22   325.7 3395.62
   333.7 3395.99   337.8 3396.89   347.9 3400.61   362.2 3409.95   367.7  3412.5
   396.1 3420.93   410.2 3426.98   428.2 3433.62   446.2  3442.1   466.1 3445.29
#Mann= 3 ,-1,0
       0      .1       0   269.5    .045       0   295.6      .1       0
#XS Ineff= 2 , 0
          163.38  3408.8
Permanent Ineff=
       F       F
Bank Sta=269.5,295.6
XS Rating Curve= 0 ,0
Exp/Cntr(USF)=0,0
Exp/Cntr=0.3,0.1

Type RM Length L Ch R = 1 ,8637    ,190.7,190,185.7
XS GIS Cut Line= 2
2154226.89811354 444622.027580812154554.03870296444816.660220512
#Sta/Elev= 30
       0  3402.7     9.1 3401.75    24.8 3398.44    38.7 3392.75    52.7 3388.03
    57.3 3386.89    71.3 3388.51    85.3 3387.68   103.9 3387.33   122.5 3387.89
   139.2 3387.49   163.7 3389.08   173.7 3389.26   178.4 3389.16193.93243386.516
     197  3386.2   204.6 3386.19213.12923386.627     263 3388.71   271.4 3391.54
   277.5 3393.07   287.8 3397.46   295.1 3400.06   299.4 3402.03   303.4 3402.89
   311.3 3403.88   322.6 3406.07   335.9 3409.82   355.2 3416.14   380.7 3425.77
#Mann= 3 ,-1,0
       0      .1       0193.9324    .045       0213.1292      .1       0
#XS Ineff= 1 ,-1
  103.23  103.23 3402.19
Permanent Ineff=
       F
Bank Sta=193.9324,213.1292
XS Rating Curve= 0 ,0
Exp/Cntr(USF)=0,0
Exp/Cntr=0.3,0.1

Type RM Length L Ch R = 1 ,8446    ,251.6,259.1,266.6
XS GIS Cut Line= 2
2154144.04098044 444824.588542182154533.63626033444918.732388733
#Sta/Elev= 30
       0 3397.69     8.4 3397.17    16.6 3395.55    24.8 3395.71    56.9 3392.77
    70.1 3390.22    74.2 3388.69    86.8 3386.11    94.8 3386.02     103 3385.15
   107.1 3385.89   113.3 3386.06   119.5 3385.03   123.2 3383.82   129.9 3383.54
   135.9 3383.84   148.3 3385.04   164.7 3384.68   177.1 3386.59   189.8  3385.1
   222.4 3387.16   239.2 3385.48     247 3386.87   255.8 3387.31   265.3  3390.5
   276.1 3397.27   292.3 3403.57   337.6 3417.78     387 3435.77   400.8    3440
#Mann= 4 ,-1,0
       0     .12       0   123.2    .045       0   135.9     .12       0
     150      .1       0
#XS Ineff= 2 , 0
          100.85 3397.69
Permanent Ineff=
       F       F
Bank Sta=123.2,135.9
XS Rating Curve= 0 ,0
Exp/Cntr(USF)=0,0
Exp/Cntr=0.3,0.1

Type RM Length L Ch R = 1 ,8187    ,127.6,139.9,147.7
XS GIS Cut Line= 2
2154037.81280342444914.0245952042154324.36444487445173.558802016
#Sta/Elev= 30
       0  3393.3    34.5 3387.73    46.4 3383.74    70.2 3378.45    76.2 3378.84
    82.2 3380.35    88.1 3380.89   111.5 3380.22   128.5 3381.08   141.7 3380.26
   159.7 3380.09   168.2 3380.85   183.5 3380.79   202.9  3382.3   231.1 3382.88
     243 3384.44   266.9  3382.3   272.8  3380.9   289.2 3380.02   295.6  3380.3
   298.4 3381.08   301.3 3382.59   305.4 3385.81   321.6 3402.84   326.7 3406.24
   338.1 3409.69   362.2  3419.5   374.9 3423.92   380.5 3425.78   386.6 3426.96
#Mann= 3 ,-1,0
       0      .1       0   272.8    .045       0   298.4      .1       0
#XS Ineff= 2 , 0
          123.49 3390.11
Permanent Ineff=
       F       F
Bank Sta=272.8,298.4
XS Rating Curve= 0 ,0
Exp/Cntr(USF)=0,0
Exp/Cntr=0.3,0.1

Type RM Length L Ch R = 1 ,8047    ,205.7,215.7,215
XS GIS Cut Line= 3
2153977.78695355444963.801251445 2154118.0011931445126.049157207
2154144.04098044445273.274108732
#Sta/Elev= 30
       0 3391.11    11.2 3389.16    28.1 3384.99    42.4 3382.44    49.4 3380.65
    65.1 3378.56    70.9 3377.24    90.6 3377.88   102.3 3377.75   113.8 3379.27
     134 3377.59   167.2 3379.23     187 3379.76   192.1 3379.47   214.4 3381.38
   225.5 3380.66   232.8 3378.66     242 3378.02   258.2 3377.98   262.3 3378.52
   274.5  3381.4   290.7 3382.99   294.8 3383.82   302.9 3386.34   329.5 3392.23
   339.5 3393.59   343.5 3393.21   347.6 3393.75   351.7 3394.89   363.9 3396.01
#Mann= 4 ,-1,0
       0     .12       0      20      .1       0   232.8    .045       0
   262.3      .1       0
Bank Sta=232.8,262.3
XS Rating Curve= 0 ,0
Exp/Cntr(USF)=0,0
Exp/Cntr=0.3,0.1

Type RM Length L Ch R = 1 ,7832    ,211.1,193.7,175.4
XS GIS Cut Line= 3
2153927.71043943444985.8349176592153941.73186338445155.093535399
2154122.00731423445277.280229862
#Sta/Elev= 30
       0 3395.12    11.4 3390.91    15.4 3388.69    23.4 3383.35    27.4 3381.26
    31.5 3379.61    39.5 3377.12    43.5 3376.63    47.5 3377.07    67.6 3376.27
    75.6 3374.88    81.9 3372.61    83.6 3371.85    87.6 3371.76    99.7 3372.46
   107.7 3372.48   111.7 3373.12   115.7 3374.41   147.8  3377.9   192.1 3376.77
   216.3 3376.78   294.8 3382.07   301.9 3382.28   312.9 3380.09   316.1 3380.03
   330.4 3383.08   346.7 3385.52   360.3 3388.06   371.8 3389.36   387.6 3392.42
#Mann= 4 ,-1,0
       0     .12       0      10      .1       0    81.9    .045       0
   107.7      .1       0
Bank Sta=81.9,107.7
XS Rating Curve= 0 ,0
Exp/Cntr(USF)=0,0
Exp/Cntr=0.3,0.1

Type RM Length L Ch R = 1 ,7638    ,182.4,190.6,186.7
XS GIS Cut Line= 3
2153719.39214067445151.0874142692153874.62933446445203.166988958
2154069.92773954445316.339910878
#Sta/Elev= 30
       0 3404.89    13.5 3395.82    17.7 3392.37    31.7 3378.83    38.8 3372.85
      43 3370.57    47.2 3369.32    68.3 3368.89    74.9 3369.32    84.4 3369.54
    93.6 3372.52      97  3372.9   119.8 3373.15   132.3 3375.44   140.1 3376.11
   148.5 3375.54   157.5 3375.93   170.1 3374.83     184 3374.83   202.5 3373.42
   211.8 3373.68   239.4 3372.25   263.5 3372.62   285.7  3374.4   318.1 3375.09
   330.3 3377.18   344.9 3382.49   359.5 3386.11   375.2 3388.54   389.5 3389.66
#Mann= 4 ,-1,0
       0     .06       0    47.2    .045       0    74.9     .06       0
      80      .1       0
#XS Ineff= 2 , 0
                          138.89         3383.82
Permanent Ineff=
       F       F
Bank Sta=47.2,74.9
XS Rating Curve= 0 ,0
Exp/Cntr(USF)=0,0
Exp/Cntr=0.3,0.1

Type RM Length L Ch R = 1 ,7447    ,221.3,206.7,196.1
XS GIS Cut Line= 3
 2153668.3440738445315.5123163252153847.58801683445380.437848957
2154039.88183107445447.540377883
#Sta/Elev= 30
       0 3400.59    12.6 3391.67    16.8 3388.19      23 3384.05    42.4 3372.92
    46.6 3371.32    55.1 3369.31    80.7 3365.3886.434013364.962   114.7  3364.3
123.00673364.619   131.7 3365.94     136 3368.44   140.2 3370.33   144.8 3370.55
   188.6 3369.11   263.3 3367.96   267.5 3367.46   276.5 3364.87   280.2 3364.32
   282.8 3364.53   292.9 3366.32   301.4  3370.5   309.9 3371.74   318.4 3375.15
   331.1 3377.02   339.5 3379.83   373.4 3387.39   390.4 3393.38   394.3 3394.39
#Mann= 4 ,-1,0
       0     .06       0      30      .1       086.43401    .045       0
123.0067      .1       0
#XS Ineff= 2 , 0
                             155         3384.48
Permanent Ineff=
       F       F
Bank Sta=86.43401,123.0067
XS Rating Curve= 0 ,0
Exp/Cntr(USF)=0,0
Exp/Cntr=0.3,0.1

Type RM Length L Ch R = 1 ,7241    ,199.1,224.7,237.1
XS GIS Cut Line= 3
2153657.29726316445566.7224814992153852.59566824445495.613831443
2154052.90172474445495.613831443
#Sta/Elev= 30
       0 3382.68    20.1 3383.51    25.3 3382.24    41.4 3377.11    45.6 3374.33
    58.4 3362.33    62.7  3360.2    66.9  3359.4    81.5 3358.81    93.9 3359.51
   109.3 3363.17     118 3364.63   122.3 3364.81   160.6 3363.57   164.8 3363.72
   173.3  3365.8   194.6 3366.87   247.4 3364.61   259.4 3365.31   279.4 3363.31
   299.4 3363.21   303.4 3363.79   307.4 3364.91   327.4  3372.5   335.4 3375.93
     345 3378.84   355.4 3382.84   397.9 3395.53   403.4 3397.28   408.1 3399.39
#Mann= 3 ,-1,0
       0      .1       0    66.9    .045       0    93.9      .1       0
#XS Ineff= 2 , 0
                          198.42         3377.44
Permanent Ineff=
       F       F
Bank Sta=66.9,93.9
XS Rating Curve= 0 ,0
Exp/Cntr(USF)=0,0
Exp/Cntr=0.3,0.1

Type RM Length L Ch R = 1 ,7016    ,217.5,276,235.1
XS GIS Cut Line= 3
 2153612.2524485445681.2987482172153770.00248601445698.426719652
2153977.49310768 445804.36698029
#Sta/Elev= 30
       0 3373.67      20 3371.76    36.1 3370.22    43.4 3368.34    48.2 3366.25
    52.2 3365.47    72.3  3362.2    88.4 3360.18     116    3360   132.7 3361.05
   148.8 3360.95   158.7 3360.28   165.6 3358.65   186.1  3356.7   212.9 3355.41
   233.7    3355   259.9 3355.57   268.9 3357.44   281.3 3357.49   296.7 3357.06
     311 3354.87   322.8  3355.9   327.3 3356.95   334.8  3359.3   340.8  3362.1
   349.7 3368.81   358.6  3373.7   364.5 3377.98   381.2 3394.51   391.6 3403.62
#Mann= 5 ,-1,0
       0      .1       0      20     .12       0   212.9    .045       0
   259.9     .12       0  298.68      .1       0
#XS Ineff= 2 , 0
                          277.11         3369.45
Permanent Ineff=
       F       F
Bank Sta=212.9,259.9
XS Rating Curve= 0 ,0
Exp/Cntr(USF)=0,0
Exp/Cntr=0.3,0.1

Type RM Length L Ch R = 1 ,6740    ,145.7,145.3,145.2
XS GIS Cut Line= 3
2153595.20238564 445781.049961952153685.34011107445880.201459916
2153778.48242734446029.429472005
#Sta/Elev= 30
       0 3367.89    14.9  3367.2    21.8 3366.03    43.3  3359.3      49  3356.8
    60.2    3350    66.9 3348.24    84.7  3347.3    94.2 3348.29    97.5 3348.93
   108.3 3352.75   114.4 3353.84   119.1 3353.73   125.4 3352.59   149.3 3352.84
   191.7 3347.81   206.4 3351.11   210.6 3352.48   215.2 3354.81     221 3358.96
   234.2 3370.44   238.9 3373.71   245.1  3376.7     253 3378.82   271.9 3381.85
     286 3386.61   290.8 3387.32   302.2 3385.77   304.9 3385.86   309.9 3387.21
#Mann= 4 ,-1,0
       0     .12       0    66.9    .045       0    94.2     .12       0
     134      .1       0
#XS Ineff= 2 , 0
                          149.07          3367.4
Permanent Ineff=
       F       F
Bank Sta=66.9,94.2
XS Rating Curve= 0 ,0
Exp/Cntr(USF)=0,0
Exp/Cntr=0.3,0.1

Type RM Length L Ch R = 1 ,6595    ,188.6,182.5,172.9
XS GIS Cut Line= 3
 2153448.9789644445838.1371880512153566.15800745445964.330003644
2153709.37683785446045.453956525
#Sta/Elev= 30
       0 3378.45     7.2 3376.56    12.9  3374.2      26 3366.05      40  3358.2
    51.7  3352.4    58.7 3349.55    63.5 3348.29    66.7 3348.15      78 3348.41
      87 3349.61    92.2 3349.57   113.3  3346.3   120.5 3344.21   135.2 3343.74
   145.8 3344.44   162.4 3348.75   165.7 3348.84   183.1 3347.45   192.9 3343.69
   198.3 3342.51   206.6 3344.06   215.9 3344.54   225.1 3348.34   238.9 3352.13
   275.7 3355.73   289.5 3356.53   307.8 3358.66   315.2 3360.48   336.8 3368.28
#Mann= 5 ,-1,0
       0     .06       0      60     .12       0      70      .1       0
   120.5    .045       0   145.8      .1       0
#XS Ineff= 2 , 0
                          183.97         3359.96
Permanent Ineff=
       F       F
Bank Sta=120.5,145.8
XS Rating Curve= 0 ,0
Exp/Cntr(USF)=0,0
Exp/Cntr=0.3,0.1

Type RM Length L Ch R = 1 ,6412    ,219,219.4,215.1
XS GIS Cut Line= 2
 2153334.8045122446046.4554868082153663.44439103446123.495327448
#Sta/Elev= 30
       0 3374.25    13.7 3369.72    26.1 3364.64    33.4 3361.03    54.8 3348.19
    71.3 3340.3975.655613338.895    83.6 3338.6793.229163339.204   103.3 3340.07
   112.3 3342.78   116.4 3343.04   128.8  3343.3   153.4 3342.51   165.7 3343.43
   183.1 3343.13   202.7 3344.11   206.8 3343.76   223.3 3339.01   239.7 3338.28
   243.8 3338.85   247.9  3340.7     252  3344.8   256.1 3346.92   284.9 3349.43
   301.3 3351.73   309.5 3354.49   317.8 3355.58     326 3357.57   337.5 3363.19
#Mann= 4 ,-1,0
       0     .12       075.65561    .045       093.22916     .12       0
     270      .1       0
#XS Ineff= 2 , 0
                          190.28            3354
Permanent Ineff=
       F       F
Bank Sta=75.65561,93.22916
XS Rating Curve= 0 ,0
Exp/Cntr(USF)=0,0
Exp/Cntr=0.3,0.1

Type RM Length L Ch R = 1 ,6193    ,168.1,168,165.9
XS GIS Cut Line= 2
2153323.78767909446269.7967398012153677.32786881446290.828875733
#Sta/Elev= 30
       0 3359.74    16.4 3359.36    28.4 3357.88    37.6 3357.23    64.5 3353.79
    68.5 3351.94    76.5 3347.46    80.5 3344.44    88.5 3336.83    92.6 3333.78
    96.6 3332.83   116.6 3331.58   139.7  3332.7   168.7  3333.9   184.7 3333.15
   192.7 3334.49   200.7 3336.57   212.8 3336.37   224.8 3337.69   232.8 3337.98
   238.1 3339.78   253.2  3346.6   275.9  3359.5   284.9 3364.95     295 3370.18
   304.9 3374.83     325 3380.85     337 3381.97     349 3384.69   354.2 3386.41
#Mann= 5 ,-1,0
       0      .1       0      60     .12       0      80      .1       0
    96.6    .045       0   139.7      .1       0
#XS Ineff= 2 , 0
                          175.12         3358.73
Permanent Ineff=
       F       F
Bank Sta=96.6,139.7
XS Rating Curve= 0 ,0
Exp/Cntr(USF)=0,0
Exp/Cntr=0.3,0.1

Type RM Length L Ch R = 1 ,6025    ,226.3,242.3,254.4
XS GIS Cut Line= 3
2153257.68668045446369.949768049 2153391.8917383446441.058418105
2153591.19626451446445.064539235
#Sta/Elev= 30
       0 3355.19     7.3 3354.85    16.1 3353.62    34.5 3350.27    39.7  3348.8
    51.6 3343.81    69.3 3338.26    75.2 3337.19    97.9 3335.04   111.5 3333.11
   151.9  3334.9   160.2    3335   188.2  3334.1   196.2 3330.59  201.053329.058
   204.2 3328.33   212.2 3328.24   226.8 3329.06   232.2  3329.7   252.2 3333.99
   256.2 3334.53   264.2 3334.57   268.2 3336.17   272.2 3338.81   280.2 3344.62
   288.2 3351.25   304.2 3361.72   328.2 3370.91   344.5 3375.37   351.2  3377.7
#Mann= 5 ,-1,0
       0     .12       0      10      .1       0  201.05    .045       0
   226.8      .1       0  261.88     .12       0
#XS Ineff= 2 , 0
          162.19 3340.24
Permanent Ineff=
       F       F
Bank Sta=201.05,226.8
XS Rating Curve= 0 ,0
Exp/Cntr(USF)=0,0
Exp/Cntr=0.3,0.1

Type RM Length L Ch R = 1 ,5782    ,191.2,190.7,189.4
XS GIS Cut Line= 3
2153215.62240858446449.0706603652153323.78767909446581.272657653
2153422.93917706446740.515972567
#Sta/Elev= 30
       0 3357.95    10.5 3354.77    13.5 3353.32    40.3 3338.22    51.6 3333.92
      57 3332.94    67.3 3332.34    76.7 3333.06      88 3332.76    98.3 3330.54
   105.6    3328   111.3 3327.21   128.4 3328.82   139.8 3328.37   159.7 3330.74
   184.8 3330.88   200.1 3328.06   208.8 3327.88   222.5 3326.29   234.9 3323.16
   243.6 3322.27   252.3 3323.02   262.4 3323.17   269.8 3324.39   279.1 3329.64
   283.8 3330.94   310.4 3333.47     338  3334.3   345.6 3336.02   358.4 3340.57
#Mann= 5 ,-1,0
       0      .1       0      30     .12       0   234.9    .045       0
   262.4     .12       0  280.81      .1       0
#XS Ineff= 2 , 0
          181.16 3339.88
Permanent Ineff=
       F       F
Bank Sta=234.9,262.4
XS Rating Curve= 0 ,0
Exp/Cntr(USF)=0,0
Exp/Cntr=0.3,0.1

Type RM Length L Ch R = 1 ,5592    ,197.1,197.1,196.5
XS GIS Cut Line= 3
2153072.40357819446605.309384432 2153180.5688487 446713.47465494
2153285.72952836446857.695015618
#Sta/Elev= 30
       0 3365.28    16.6 3358.47    25.2 3353.73    39.3 3344.82    45.1 3340.69
    50.7 3337.35    56.4 3333.36    73.2 3323.86    78.9 3323.06    84.5 3323.15
   101.6 3324.57   118.6 3324.63     144 3325.49   152.6 3326.29   157.6 3326.26
   163.9 3325.49   182.3 3320.28   186.8 3319.36   197.2 3319.08     217 3319.51
   241.7 3322.96   247.3 3324.89   256.6 3326.54   264.1 3326.82   272.7  3327.7
   281.4 3327.66   288.1 3328.27   307.1 3328.83   325.9 3330.55   331.5 3331.52
#Mann= 5 ,-1,0
       0     .06       0      40     .12       0   186.8    .045       0
     217     .12       0  222.97      .1       0
#XS Ineff= 2 , 0
          158.52 3333.34
Permanent Ineff=
       F       F
Bank Sta=186.8,217
XS Rating Curve= 0 ,0
Exp/Cntr(USF)=0,0
Exp/Cntr=0.3,0.1

Type RM Length L Ch R = 1 ,5395    ,265.6,245.7,235.1
XS GIS Cut Line= 3
2152981.26432248446779.5756535842153106.45560779446939.820498781
2153243.66525649446970.867937538
#Sta/Elev= 30
       0 3342.86    17.5 3331.41    30.7  3323.9    34.6  3322.2    42.6 3319.98
    52.8 3318.36    63.2 3319.17    80.2 3321.38   100.1 3320.93   105.8 3319.99
   115.2 3316.31   131.5 3315.95   147.7 3316.23   162.8 3319.84   168.5 3320.77
   184.8 3320.72     200 3321.87   221.5 3320.51   229.7 3320.31   239.4 3320.71
   250.2 3320.47   262.5 3321.31   266.6 3321.28   270.7 3320.79   274.8 3319.59
   278.9 3320.39     283 3322.33   295.3 3325.19   332.2 3335.54     344 3337.11
#Mann= 5 ,-1,0
       0      .1       0      40     .12       0     110      .1       0
   115.2    .045       0   147.7      .1       0
#XS Ineff= 2 , 0
           85.55 3326.67  200.54         3327.16
Permanent Ineff=
       F       F
Bank Sta=115.2,147.7
XS Rating Curve= 0 ,0
Exp/Cntr(USF)=0,0
Exp/Cntr=0.3,0.1

Type RM Length L Ch R = 1 ,5149    ,306.4,312.8,306.6
XS GIS Cut Line= 2
2152843.49094757447065.8993337162153225.27188644447143.586903698
#Sta/Elev= 30
       0 3341.68      17 3339.27    29.3 3331.46      53 3318.0364.354793313.081
    70.1 3311.75    90.5 3311.58    98.7 3311.85   105.1 3312.77   119.1 3314.52
   152.6    3315   176.2 3314.53     213 3314.57   220.4  3313.7   237.1 3314.84
   253.8 3314.61     258 3314.06   271.3 3314.34   282.4 3315.17   294.6 3314.12
   306.8 3315.05   323.2 3317.67   327.3  3318.8   331.3 3320.53   339.5 3325.41
   347.7 3331.76   351.7 3335.83   368.1 3347.49   380.3 3353.76   389.6  3356.3
#Mann= 3 ,-1,0
       0      .1       064.35479    .045       0   105.1      .1       0
#XS Ineff= 1 ,-1
  123.94   383.1 3323.85
Permanent Ineff=
       F
Bank Sta=64.35479,105.1
XS Rating Curve= 0 ,0
Exp/Cntr(USF)=0,0
Exp/Cntr=0.3,0.1

Type RM Length L Ch R = 1 ,4836    ,246.3,257.3,261.3
XS GIS Cut Line= 3
2152809.15709612447229.7964991022152966.24136824447329.415778667
2153087.42653243447390.509125898
#Sta/Elev= 30
       0 3321.22    24.9 3316.96    39.4 3315.37    48.1 3315.36    55.7 3316.24
    58.6 3316.24    77.1 3311.89    82.9 3311.43    91.6 3312.33    97.4 3311.92
   112.5 3308.55   118.3  3308.2   129.3  3308.3   143.8 3307.28   164.6    3310
   170.6 3310.08   178.1 3309.46   193.2 3309.98     223 3307.89238.76193304.805
   241.9  3304.4   250.9 3304.22   255.4 3304.59256.56193305.006   261.7 3307.09
   276.6 3314.31   291.2 3324.92   304.6 3333.13   313.6 3338.08   321.7 3341.19
#Mann= 4 ,-1,0
       0     .12       0     120      .1       0238.7619    .045       0
256.5619      .1       0
#XS Ineff= 2 , 0
          168.28 3316.66
Permanent Ineff=
       F       F
Bank Sta=238.7619,256.5619
XS Rating Curve= 0 ,0
Exp/Cntr(USF)=0,0
Exp/Cntr=0.3,0.1

Type RM Length L Ch R = 1 ,4579    ,198.4,196.3,193.2
XS GIS Cut Line= 2
 2152728.8786913447303.3759913222152874.10058226447526.717244316
#Sta/Elev= 30
       0 3328.62    20.7 3324.06      26 3322.59    41.3  3316.9    50.1 3313.02
    64.2 3308.16    72.1 3307.06    78.5 3305.66    83.3 3305.35   102.3 3300.03
   107.8 3299.17   113.6 3297.81   121.4 3297.33   130.8 3297.89   140.5  3298.9
   154.8 3302.72   159.6 3302.91   164.4 3302.14   169.1 3302.01   171.4 3302.78
   174.3 3304.33   182.2 3309.08   191.6 3315.28   200.3 3320.08   207.3 3324.59
   212.1 3326.89   226.2 3331.08     235 3333.11   250.3 3335.64   266.4 3337.86
#Mann= 4 ,-1,0
       0     .12       0   113.6    .045       0   130.8     .12       0
     140      .1       0
Bank Sta=113.6,130.8
XS Rating Curve= 0 ,0
Exp/Cntr(USF)=0,0
Exp/Cntr=0.3,0.1

Type RM Length L Ch R = 1 ,4383    ,208.1,199.3,189.9
XS GIS Cut Line= 2
2152579.65067921447457.6116548252152735.88940327447627.871802846
#Sta/Elev= 30
       0 3333.81    11.4 3330.76    24.4 3326.54    42.2 3318.54    48.2 3315.28
    53.9 3311.56    59.9 3305.72    62.3 3304.06    75.4 3296.26    79.3 3294.59
    83.6 3294.17    95.4 3294.03   107.3 3294.52   124.6 3298.05   127.5  3298.4
   130.3 3298.53   136.8  3297.9   140.6 3297.83   152.9 3298.09   155.8 3298.43
   161.4 3299.69   167.1 3300.57   173.1 3301.05   189.7 3300.86   194.9 3301.33
   201.9 3302.52   205.7 3303.56   212.4 3306.68   225.6 3314.73   231.1 3316.42
#Mann= 5 ,-1,0
       0      .1       0      50     .12       0    79.3    .045       0
   107.3     .12       0     130      .1       0
Bank Sta=79.3,107.3
XS Rating Curve= 0 ,0
Exp/Cntr(USF)=0,0
Exp/Cntr=0.3,0.1

Type RM Length L Ch R = 1 ,4183    ,291.5,293.5,290.1
XS GIS Cut Line= 2
2152439.43643966447664.9284232982152731.88328214447756.067679004
#Sta/Elev= 30
       0 3326.21    13.3 3321.49      20 3319.76    34.3  3315.1    43.3 3312.73
    63.6 3308.83    67.8 3307.14    80.4 3300.89    92.9 3292.18    97.1 3289.76
    99.8 3289.32   118.1 3288.78     119 3288.92   143.2 3292.95   147.4 3293.26
   163.7 3293.55   172.6 3291.12   176.5  3292.1   180.9 3294.21   189.3 3297.19
   211.6 3296.88     248 3298.08   252.2 3298.74   256.3 3299.73   260.5 3301.94
   273.1 3310.57   285.7 3320.24   289.9 3321.94   294.1 3323.04   306.3 3328.17
#Mann= 3 ,-1,0
       0      .1       0    99.8    .045       0     119      .1       0
#XS Ineff= 2 , 0
                          161.29          3303.3
Permanent Ineff=
       F       F
Bank Sta=99.8,119
XS Rating Curve= 0 ,0
Exp/Cntr(USF)=0,0
Exp/Cntr=0.3,0.1

Type RM Length L Ch R = 1 ,3890    ,115.6,117,117.3
XS GIS Cut Line= 3
2152278.19006418447838.1931621682152440.43796994447886.266615727
2152690.82054056447874.248252337
#Sta/Elev= 30
       0 3325.35    13.7 3317.24    39.6 3296.98    43.8 3292.97    52.1 3283.17
    56.3 3281.91    68.8 3281.36    77.2 3279.86    89.7 3281.32   102.2    3285
   114.7 3287.68   139.7 3287.26   156.4 3288.47     185 3289.09     205 3290.69
     217 3289.07     229 3288.72     237 3289.27     249    3291   277.1    3292
   293.1 3293.76   297.1 3295.74   313.1 3305.46   325.1  3310.2   345.8 3319.72
   364.9 3326.77   380.2  3331.3   389.2 3334.85   405.2 3342.54   419.9 3347.99
#Mann= 3 ,-1,0
       0      .1       0    68.8    .045       0    89.7      .1       0
Bank Sta=68.8,89.7
XS Rating Curve= 0 ,0
Exp/Cntr(USF)=0,0
Exp/Cntr=0.3,0.1
